HEC-RAS study CaneyFork.prj: Caney Fork River- Smith County

--- CaneyFork.g02 (geometry) --- (continued)

Type RM Length L Ch R = 1 ,60398.76,113.4,185.5,277.1
BEGIN DESCRIPTION:
18843.96
END DESCRIPTION:
XS GIS Cut Line= 6
      1993727.33        674212.5      1994680.87       674390.22
  1996262.187807674342.226877199      1997778.05       673621.94
      1998388.06       673642.98      1999209.16       673037.55
#Sta/Elev= 30
       0  609.35   141.6  576.72     279  555.42   652.8  518.78   952.9  517.97
  1148.3  506.48  1188.4  499.16    1471  527.31  2099.8  532.84  2229.6  490.73
  2422.7  485.42 2589.11  467.64 2617.51  459.59    2688  448.96 2856.86  460.19
    2956   493.3  3291.3  497.06  3629.6  515.72  3851.3  512.62  4046.5  540.87
  4146.4  540.39  4315.9  581.39    4581  698.89  4733.6   725.5  4818.7  721.38
    4949  703.08  5083.1  674.55    5294  640.29  5477.6  635.95  5862.9  598.08
#Mann= 3 , 0 , 0
       0      .1       0 2617.51    .035       0 2856.86      .1       0
Bank Sta=2617.51,2856.86
XS Rating Curve= 0 ,0
Exp/Cntr=0.5,0.3

Type RM Length L Ch R = 1 ,60213.25,98.6,102.3,100.2
BEGIN DESCRIPTION:
18775.39
END DESCRIPTION:
XS GIS Cut Line= 6
      1993699.93        674247.51994732.34832747  674434.3331228
1996747.53709946674444.817807001      1998024.93       673987.58
      2000384.35       673216.72      2002345.02       673046.43
#Sta/Elev= 30
       0 610.771 298.915 554.291 707.952 518.0431215.914 502.8121495.926 527.143
2150.956 531.9062298.463 488.7182669.026 470.125 2717.19  453.03 2816.96  450.69
 2940.78 470.0993087.333 496.4043642.298 493.7213899.865 521.1524213.194 568.036
 4509.74 693.1114630.722 711.8934766.406 708.0365238.263 638.9285498.638 676.147
 5632.77 677.2936340.252 551.5216816.291 626.8537128.943 695.6757437.601 736.514
7630.826 737.9867881.767 710.4188325.933 620.7038694.816 716.4868871.432 742.543
#Mann= 3 , 0 , 0
       0      .1       02669.026    .035       0 2940.78      .1       0
Bank Sta=2669.026,2940.78
XS Rating Curve= 0 ,0
Exp/Cntr=0.5,0.3

Type RM Length L Ch R = 3 ,60139.2 ,,,
Bridge Culvert--1,0,-1,-1, 0
Deck Dist Width WeirC Skew NumUp NumDn MinLoCord MaxHiCord MaxSubmerge Is_Ogee
28,29,2.61,0, 15, 15, , , 0.95, 0, 0,0,,
 2403.47    2475 2616.62 2616.63 2622.26 2627.72 2631.74 2713.72 2799.52  2885.4
 2970.49 3071.163071.161 3153.73  3329.3
  490.93  492.22     491  492.95  494.05  494.05  494.05  494.05  494.59  494.94
  495.43  496.86   491.7   495.5  495.92
                                          452.72  485.88  486.55  487.09  487.44
  487.93
    2300    2325    2525 2683.21 2683.21 2688.71 2695.02 2777.31 2862.09  2946.5
 3032.09 3127.223127.221 3203.73  3979.3
  490.93  492.92  492.22     491  494.41  495.47  495.47  495.47   494.6  495.03
  495.45  495.93   491.7   495.5  495.92
                                                  486.51  486.79   487.1  487.53
  487.95
Pier Skew, UpSta & Num, DnSta & Num=  ,2713.72, 2 ,2777.31, 2 , 2 , 2 , 0 ,,
      .4      .6
  470.11  486.55
      .4      .6
  470.11  486.79
Pier Skew, UpSta & Num, DnSta & Num=  ,2799.52, 2 ,2862.09, 2 , 2 , 2 , 0 ,,
      .4      .6
  450.63  487.09
      .4      .6
  450.63   487.1
Pier Skew, UpSta & Num, DnSta & Num=  ,2885.4, 2 ,2946.5, 2 , 2 , 2 , 0 ,,
      .4      .6
  453.87  487.44
      .4      .6
  453.87  487.53
Pier Skew, UpSta & Num, DnSta & Num=  ,2969.49, 2 ,3032.09, 2 , 2 , 2 , 0 ,,
      .4      .6
   467.4  487.93
      .4      .6
   467.4  487.95
BR Coef=-1 , 0 , 0 ,, 0 ,,,0.8,0,,0,
WSPro=,,,, 1 ,,,, 0 ,,,, 0 ,,,,-1 ,-1 ,-1 , 0 , 0 , 0 , 0 , 0
BC Design=,, 0 ,, 0 ,,,,,,
BC HTab HWMax=600
BC Use User HTab Curves=0
BC User HTab FreeFlow(D)= 0

Type RM Length L Ch R = 1 ,60110.92,921.8,922.8,879.3
XS GIS Cut Line= 6
1993695.15939903674283.8345869961994734.41239648674484.151886339
 1996326.6781092674540.6516374361996752.04323867 674541.03210714
2000394.73802469673287.5666925752002340.28879151673128.095318245
#Sta/Elev= 30
       0 606.793 278.949 555.297  693.95 520.9691255.661 505.031 1508.32 526.042
2181.243 531.4362348.849  487.072686.539 474.997 2760.19  453.03 2859.96  450.69
3033.427 476.3453132.033   494.13578.847 490.7553959.564 522.7944234.527 565.148
4477.387 662.3984562.367 685.4314652.258 693.4054935.152 668.4185218.046 614.411
5508.381 665.622 5664.86 674.9896042.934 599.7896403.372 545.5967184.522 685.415
 7498.07 724.9727799.076 706.7828376.004 616.2938707.111 700.4188881.415 719.578
#Mann= 3 , 0 , 0
       0      .1       02686.539    .035       03033.427      .1       0
Bank Sta=2686.539,3033.427
XS Rating Curve= 0 ,0
Exp/Cntr(USF)=0,0
Exp/Cntr=0.5,0.3

Type RM Length L Ch R = 1 ,59188.11,1292,1615.6,1754.8
BEGIN DESCRIPTION:
18473.60
END DESCRIPTION:
XS GIS Cut Line= 6
      1993752.94        674471.31996395.67756006675445.466062076
      2000910.27       676719.53      2001749.79       676178.82
       2003684.2       676615.63      2006599.02       676709.57
#Sta/Elev= 30
       0  572.36   407.9  531.19  1282.1  502.84  1620.1  528.76  2280.7  522.44
  2663.7  507.32 3004.27  460.53  3124.2  450.01 3342.72  460.45  3407.9  481.86
  3545.7  488.32    4046  470.23  4308.3  500.39  4871.5  497.56  5321.1  539.07
  6024.6  656.04  7111.4  674.89  7900.5     720  8361.4  788.84  9393.5  881.62
    9635  893.41   10042  869.29 10776.9  977.54 10877.8   965.3 11025.4  882.07
 11190.5  851.59 11860.9  627.71   12116   602.6 12368.3  632.28 13496.7  831.88
#Mann= 3 , 0 , 0
       0      .1       0 3004.27    .035       0 3342.72      .1       0
Bank Sta=3004.27,3342.72
XS Rating Curve= 0 ,0
Exp/Cntr=0.3,0.1

Type RM Length L Ch R = 1 ,57572.5 ,1665.9,1810.1,1959.5
BEGIN DESCRIPTION:
17986.65
END DESCRIPTION:
XS GIS Cut Line= 6
       1992412.6       674476.31      1993521.95       674952.96
      1993961.08       675321.551996296.51536002676666.726841486
      1998818.21       678816.28      2000604.69       681142.87
#Sta/Elev= 30
       0  731.69     505  657.38   913.1  644.85  1370.6  555.76    1752  509.65
  2295.7  496.75  2792.3  529.15  4454.4  493.36  4519.9  469.57    4660  468.72
  4743.5  444.12  4853.4  469.16  4954.8   498.5  4964.6  584.74  4979.4  610.88
  5051.1   672.7  5098.7   684.9  5443.5  649.71  6198.8  629.68    6772  671.04
  7250.2  804.24  7628.2  874.52  7762.8  867.29  8054.7  894.14  8423.5  862.19
  8804.9  892.41  9156.8  852.06  9590.4  921.96  9961.6  887.44 10724.4  912.28
#Mann= 3 , 0 , 0
       0      .1       0    4660     .05       0  4853.4      .1       0
Bank Sta=4660,4853.4
XS Rating Curve= 0 ,0
Exp/Cntr=0.3,0.1

Type RM Length L Ch R = 1 ,55762.41,2532.5,2460,2368.5
XS GIS Cut Line= 4
      1992223.05       675460.751994997.52120022677131.630171987
      1995036.46       678092.01      1996873.19       681408.32
#Sta/Elev= 30
       0  669.84   130.1  645.48     416  570.34   953.1  492.83  2262.9  504.03
  2738.6  487.21  3462.7  491.16  3592.8  480.84  3685.4  486.35  3726.1  477.27
 3874.73  444.54 3962.94  444.55 4022.57  474.53  4080.7  519.67  4085.7   574.4
  4088.2  585.03  4100.7     589  4198.5  596.18  4449.5  578.72  4512.4  584.22
    5144  695.38  5255.5  707.26  5369.8   713.3    5567  701.38  6047.4  613.77
  6407.2  560.83  6547.2  582.25  7234.2  732.65    7676  792.24  7990.9  812.86
#Mann= 3 , 0 , 0
       0      .1       0  3726.1    .045       0 4022.57      .1       0
Bank Sta=3726.1,4022.57
XS Rating Curve= 0 ,0
Exp/Cntr=0.3,0.1

Type RM Length L Ch R = 1 ,53302.41,2668.7,2677.5,2686.9
BEGIN DESCRIPTION:
16626.80
END DESCRIPTION:
XS GIS Cut Line= 5
1991589.42382875676458.7653711021992369.21211441677455.414628898
1992852.93102823678766.569027865      1993210.03       678944.96
      1994773.22       681558.12
#Sta/Elev= 30
       0  633.77   468.7  570.97   498.4  561.56   593.9  500.03   652.7  479.72
   925.8  491.99  1313.4  479.83  1691.6  491.85  1737.1  468.03  1863.2  451.15
  1948.1  449.92 2029.96  452.53 2050.57  460.11  2134.1  468.03    2286  483.81
  2581.8  483.71  2645.4  477.92  2733.1  490.42  2843.1  528.23  3120.9  528.37
  3404.5  548.51  3627.8  576.57  3990.4  608.04  4160.9  631.06  4210.4  630.66
  4462.8  667.38    4890  701.84  5224.2  711.66  5605.9  683.34  6107.2  664.87
#Mann= 3 , 0 , 0
       0      .1       0  1737.1     .04       0  2134.1      .1       0
Bank Sta=1737.1,2134.1
XS Rating Curve= 0 ,0
Exp/Cntr=0.3,0.1

Type RM Length L Ch R = 1 ,50624.91,1919.9,1839.9,1769.1
BEGIN DESCRIPTION:
15807.77
END DESCRIPTION:
XS GIS Cut Line= 6
      1990460.85       673152.28       1990420.7       674309.29
      1989353.86       677519.031989875.06372574678377.252160399
1990427.29646832679929.412216497      1991471.12       681706.82
#Sta/Elev= 30
       0  756.57   100.7  756.74   558.4  701.04  1301.1  703.31  1567.2  661.59
    1907  589.58  2465.6  539.27  2863.4   532.1  3772.3  585.65  4370.3  592.44
  5013.2  538.73  5274.4  533.54  5453.8  501.98  5548.4  497.11    5641  473.23
  5930.5  480.38  6092.4  467.72  6191.1  451.07  6305.9  446.83  6354.3  447.47
  6418.8  467.72  6469.3  490.44  7140.6  488.25  7662.8  506.72  7884.9  532.88
  8158.9  595.65  8329.9  592.26  8406.4  573.31  8808.2   688.5  9256.5  779.41
#Mann= 3 , 0 , 0
       0      .1       0  6092.4    .035       0  6418.8      .1       0
Bank Sta=6092.4,6418.8
XS Rating Curve= 0 ,0
Exp/Cntr=0.3,0.1

Type RM Length L Ch R = 1 ,48785.00,1317.7,1317.3,1313.3
XS GIS Cut Line= 4
      1986140.37       672053.65      1987350.31       678326.05
      1989436.62       681104.41      1989526.75       681904.01
#Sta/Elev= 30
       0  574.83   449.9  592.74   647.1  567.23  1063.5  602.14  1590.5  580.56
  1748.4  606.12  2320.4  613.03  2377.3  612.52  2456.2  575.32  2792.3  575.31
  2998.5  611.83  3411.1  614.38  3512.8  592.13  3841.3  585.92  3963.5  604.98
  4011.9  580.23  4205.1  572.65  5682.1  597.69  6316.1  578.95  6652.4  547.08
  6914.7  550.45  7052.1  511.95  7365.8  467.49  7981.6  499.98  8022.2  470.48
 8243.95  444.54  8379.4  469.78  9901.8  512.25 10241.5  572.46 10667.2  706.13
#Mann= 3 , 0 , 0
       0      .1       0  8022.2    .035       0  8379.4      .1       0
#XS Ineff= 2 , 0
         7981.23  499.98
Permanent Ineff=
       F       F
Bank Sta=8022.2,8379.4
XS Rating Curve= 0 ,0
Exp/Cntr=0.3,0.1

Type RM Length L Ch R = 1 ,47467.66,1886.3,1914.4,1980.5
BEGIN DESCRIPTION:
14857.42
END DESCRIPTION:
XS GIS Cut Line= 6
1979772.62082924668057.8368607941985618.17771665672428.004044132
      1985262.81       675300.72      1986685.82       676942.43
      1986545.92       679395.72      1988443.09       681868.92
#Sta/Elev= 30
       0  884.24  1247.8  713.73    2523  620.69  2759.9  630.92  3294.3  576.34
  3944.1  555.43  5420.1  554.79    5561  535.89  5879.1  591.32  6260.2  580.21
  6484.2  631.59  7022.3  638.28  7943.8   600.9  8427.2  655.91  8780.2  665.73
  9130.7  662.93    9572  592.15 10116.8  699.79 10520.9  677.55 11205.7  735.23
 13491.6  538.41 14069.3  543.16 14174.1  519.14 15890.9  493.79 16219.3  466.81
16286.25  444.54 16572.4  466.81   16834  487.85   17548   660.2 18099.7   713.7
#Mann= 3 , 0 , 0
       0      .1       0 16219.3    .035       0 16572.4      .1       0
Bank Sta=16219.3,16572.4
XS Rating Curve= 0 ,0
Exp/Cntr=0.3,0.1

Type RM Length L Ch R = 1 ,45553.31,1887.6,1827.5,1788.3
BEGIN DESCRIPTION:
14274.22
END DESCRIPTION:
XS GIS Cut Line= 6
      1973413.14       680048.95      1978737.88       679921.31
      1982888.56       678324.39      1985238.82       680632.07
      1985840.91       681709.33      1988031.57       683288.38
#Sta/Elev= 30
       0 1018.48   951.2  738.48  1348.8  678.78  2141.8  725.16  2814.2  906.89
  3134.3  942.63  3394.4  920.61  4339.7  720.38  5014.9  685.04  5322.5  710.15
  6222.2  611.22  7312.6  582.15  8297.2  617.13  8508.1  559.71  8908.9  546.22
  9648.2  749.04 10236.3  780.14 10921.9  732.42 11433.3  747.42 12685.1  488.67
 13867.6  476.62 13932.2  444.06 14181.7   474.7 14371.4  535.58 14875.9  597.52
 15460.1  607.94 15686.7  576.75 16231.6  643.09 16535.9  575.26 17017.1  667.32
#Mann= 3 , 0 , 0
       0      .1       0 13867.6    .035       0 14181.7      .1       0
Bank Sta=13867.6,14181.7
XS Rating Curve= 0 ,0
Exp/Cntr=0.3,0.1

Type RM Length L Ch R = 1 ,43725.78,1896.7,1559.3,1493.8
XS GIS Cut Line= 6
      1972201.53       680579.03      1975085.88       680323.84
      1980484.03       681114.071983538.17171434 681744.55291456
1984609.40262853682926.305599188       1986967.2       683800.21
#Sta/Elev= 30
       0  834.08   353.9   734.5     635  819.76   933.7  872.24  1167.1   895.7
  1601.3  880.62  2959.5  648.69  3626.5  742.07  4141.9  885.81  4437.6  931.64
  4745.8  888.01  5190.5  879.45  5813.1  821.71    6474  789.07  6830.3  809.64
  7785.4  638.68  8144.2  682.84  8775.1  669.35  9686.4  551.74 10341.4  558.57
 10587.5     508 11052.1   529.3 11299.7  482.95 12191.4   473.9 12269.2  446.89
12474.75  444.62 12557.5   471.1 12714.5  509.38 14053.7  513.45 15579.4  608.09
#Mann= 3 , 0 , 0
       0      .1       0 12191.4    .035       0 12557.5      .1       0
Bank Sta=12191.4,12557.5
XS Rating Curve= 0 ,0
Exp/Cntr=0.3,0.1

Type RM Length L Ch R = 1 ,42166.46,1661.7,1495.8,1288.8
BEGIN DESCRIPTION:
13144.98
END DESCRIPTION:
XS GIS Cut Line= 6
      1960814.12       690884.11      1965382.51       683560.99
      1969809.43       682427.32      1974167.64        680663.1
      1981985.32       683620.73      1986032.69       684250.52
#Sta/Elev= 30
       0  870.13   623.2  746.38  1433.5  927.68  2965.7  962.57  5582.9  738.04
  6807.3 1026.74  7880.6  710.39  8479.4  914.53  9154.1 1015.49 10774.8  636.41
 11941.3  876.05 12798.1  898.01 13281.5   994.3 13772.3  859.93   14669  767.76
 15284.9  823.47 16493.7  671.94 17229.8  737.92 17826.1   887.6 19187.5  573.26
 20625.3   782.7   21726  604.98 22368.1     691   24616  666.48 25586.3  764.61
 26835.6  545.66 27009.6   447.927321.93   470.427672.03   472.9 30501.6  584.95
#Mann= 3 , 0 , 0
       0      .1       027321.93    .035       027672.03      .1       0
Bank Sta=27321.93,27672.03
XS Rating Curve= 0 ,0
Exp/Cntr=0.3,0.1

Type RM Length L Ch R = 1 ,40670.64,1057,1047.6,1032.5
XS GIS Cut Line= 6
      1971575.33       690568.37      1974422.64       686427.82
      1979233.48       684217.831982823.88372574685007.708365676
1983854.91780669684697.896985142      1986081.16       685227.15
#Sta/Elev= 30
       0   667.2   404.5  625.67   581.4  637.27  1418.9  793.14  2414.5  647.32
  2929.8  632.51  3491.6  672.23  4657.4  936.83  5089.5  838.13  5735.7  862.38
  6140.5  828.89  6596.2  845.39  7932.5  800.92  8297.9  761.11  9249.8  571.57
  9955.6  585.81 10346.7  504.49 12598.3  500.19 13151.8  466.71 13316.7  532.72
 13451.6  491.38   13978  535.02 14069.6  486.1614153.25   445.6   14611  486.57
 15715.3  495.11   16561  535.16 16889.6  518.07 17226.3   579.9   17410  559.96
#Mann= 3 , 0 , 0
       0      .2       0 14069.6     .05       0   14611      .2       0
#XS Ineff= 2 , 0
        13320.96  533.17
Permanent Ineff=
       F       F
Bank Sta=14069.6,14611
XS Rating Curve= 0 ,0
Exp/Cntr=0.3,0.1

Type RM Length L Ch R = 1 ,39623.04,2025.5,1938.8,1779.7
XS GIS Cut Line= 5
      1979337.02       688666.83       1981704.4        687021.7
      1982988.14       686086.65 1984099.2322165685605.269348847
      1985952.59       685538.22
#Sta/Elev= 30
       0  695.36   120.8  651.63   358.2  612.58   694.7  644.49   953.2  633.32
  1482.1  571.42  1814.9  602.29  2142.7  595.74  2544.1  555.81    2704  524.76
  2888.6  574.22  3284.5  590.73    3662  569.55  3986.6  520.24    4197  503.65
    4308  513.18  4537.4  492.87  4578.3  508.11    4611   488.6  4758.1  475.06
 4796.24  454.19  4883.7  444.54 5116.94  445.51 5134.34  454.31  5202.2  475.59
  5439.3  477.98  5615.2  499.59  6031.7  485.74  6229.6  505.92  7536.5  545.92
#Mann= 3 , 0 , 0
       0      .2       0 4796.24    .045       0 5134.34      .2       0
#XS Ineff= 2 , 0
         2232.31  696.71 5767.49          501.72
Permanent Ineff=
       F       F
Bank Sta=4796.24,5134.34
XS Rating Curve= 0 ,0
Exp/Cntr=0.3,0.1

Type RM Length L Ch R = 1 ,37684.22,1311.4,1331.1,1342
BEGIN DESCRIPTION:
11729.94
END DESCRIPTION:
XS GIS Cut Line= 6
      1982336.32       690252.69      1983456.59       689713.15
      1983464.51       689145.48      1984373.47       687670.47
      1984758.11        687208.2      1986096.38        686185.8
#Sta/Elev= 30
       0  546.29    95.6  546.21   322.2   592.6     694  626.51  1071.4  605.55
  1296.2   579.8  1443.7  547.98  2397.2   526.5    2470  511.87  2770.9  508.55
  2827.8  496.21  3230.3  495.49  3307.2  490.63  3403.9  465.63  3772.2  480.31
  3831.3  465.13  3847.7   460.4  3857.1   447.8  3906.9   443.3  4043.4   448.3
  4070.6464.7505  4271.3  473.86  4375.3   466.9  4510.5  490.38  4599.2   487.6
  4928.7  563.64  5371.2  613.84  5499.1  608.61  5790.8   552.6  5867.1  548.52
#Mann= 3 , 0 , 0
       0      .2       0  3831.3     .04       0  4070.6      .2       0
Bank Sta=3831.3,4070.6
XS Rating Curve= 0 ,0
Exp/Cntr=0.3,0.1

Type RM Length L Ch R = 1 ,36353.12,1824.2,1625.1,1434.9
XS GIS Cut Line= 6
      1985143.32       690711.82        1985255.       690023.81
      1985091.83       689535.64      1985427.94       688452.77
1986263.78423894687613.524514855      1986137.99       686138.65
#Sta/Elev= 30
       0  621.62   381.4   665.1   472.5   691.1   548.5  691.51   654.9  672.75
   863.4  610.78   912.2  575.17  1001.6   538.6  1077.5  538.23  1146.7  582.34
  1294.6  577.58  1480.8  507.05    1761  489.33  2160.4  494.69  2329.2  469.88
  2483.9  464.53 2566.77  444.54 2715.16  445.13  2792.2  464.53  2887.4  486.76
  3220.8  501.84  3409.6  548.57  3546.3  564.72  4098.7  566.82  4319.8  541.48
  4447.7  560.21  4581.5  563.65  4736.3  588.05  4887.6  574.67  5026.6  546.38
#Mann= 3 , 0 , 0
       0     .15       0  2483.9    .035       0  2792.2     .15       0
Bank Sta=2483.9,2792.2
XS Rating Curve= 0 ,0
Exp/Cntr=0.3,0.1

Type RM Length L Ch R = 1 ,34728.04,1946.4,1874.4,1821.1
BEGIN DESCRIPTION:
10887.60
END DESCRIPTION:
XS GIS Cut Line= 6
      1987950.32       691170.96      1986709.21       690012.52
1987073.06993102689122.406274257      1986825.28       688243.15
      1986573.96       686738.01      1986145.15       686073.15
#Sta/Elev= 30
       0     697   350.5  823.98     470  840.23   722.6     915   938.7  913.26
    1397  870.74    1776  941.13  1924.2  894.02  2167.3  842.52  2318.5  698.92
  2408.6  631.42  2540.9  564.58  2575.1  562.05  2596.7   530.4    2690   484.2
  2766.3  468.66 2804.62  444.54 2938.85  444.54  2978.3  464.19  3585.6   489.9
  3870.6  531.25  4074.6  534.96  4300.4  514.33  4461.1     534  4644.4  530.57
  4946.8   587.4  5337.3  599.41  5681.2  578.86  5807.8  547.16    5898  545.97
#Mann= 3 , 0 , 0
       0      .1       0  2766.3    .035       0  2978.3      .1       0
Bank Sta=2766.3,2978.3
XS Rating Curve= 0 ,0
Exp/Cntr=0.3,0.1

Type RM Length L Ch R = 1 ,32853.63,1670.5,1590.4,1491.4
XS GIS Cut Line= 5
      1989624.98       689096.55       1988863.4       688357.61
      1988693.68       688129.13      1987822.35       686775.94
      1986202.52        685672.7
#Sta/Elev= 30
       0  803.12   105.8  798.09   255.6  762.91   427.6  758.67   773.6  671.39
   833.8  639.23   848.3  613.75   857.2  579.61   860.7  554.56   866.9  548.16
  1098.2  463.75 1119.58  446.56 1176.66  444.54 1319.36  445.64  1394.8  463.75
  1451.3  470.02    1493  489.94  1818.5  484.74  2111.4  505.78  2358.2  487.05
  2455.2  507.97  2732.9  494.42  3062.8  497.86  3484.7  549.37  3639.8  539.17
  3803.1  553.35    3915   541.4  4172.1  542.17  4532.1  525.63  4915.1  545.08
#Mann= 3 , 0 , 0
       0      .1       0  1098.2    .035       0  1394.8      .1       0
Bank Sta=1098.2,1394.8
XS Rating Curve= 0 ,0
Exp/Cntr=0.3,0.1

Type RM Length L Ch R = 1 ,31263.19,2954.5,2931,2891.2
BEGIN DESCRIPTION:
9747.548
END DESCRIPTION:
XS GIS Cut Line= 6
      1991194.59       688347.04      1990677.92        687318.7
      1989324.14       686744.77      1987418.98       685659.15
      1986686.21       685461.16      1986082.88       685174.04
#Sta/Elev= 30
       0  609.91   653.4  554.69   819.1  556.74  1009.1  582.91    1149  591.15
  1491.3  577.83  1902.1  492.12  1957.6  488.24  2068.6  495.66 2124.16  461.49
 2213.55  444.57 2302.93  444.54 2332.73  444.76 2392.32  461.57  2506.3  476.19
  2614.5  475.44  2690.6  485.82    2867  494.58  3454.4  480.82  3595.6  490.53
  4363.3  503.92  4524.3  516.72  4818.2   553.1  5066.8  544.13  5441.9  577.61
  5698.4  570.67  5911.5  548.91  6014.2  546.16  6164.7     549  6245.6  560.74
#Mann= 3 , 0 , 0
       0      .1       0 2124.16    .035       0 2392.32      .1       0
#XS Ineff= 2 , 0
                         2899.12          494.84
Permanent Ineff=
       F       F
Bank Sta=2124.16,2392.32
XS Rating Curve= 0 ,0
Exp/Cntr=0.3,0.1

Type RM Length L Ch R = 1 ,28332.15,1545.5,1797.3,2133.6
BEGIN DESCRIPTION:
8852.190
END DESCRIPTION:
XS GIS Cut Line= 6
      1990815.21       687236.61      1991542.08       685603.12
1991407.49896967684858.8013253091990827.65426256 684229.72191109
1990296.54617782       684051.99      1990065.13       682554.04
#Sta/Elev= 30
       0  598.88   373.1  613.53   661.9  597.04   825.5  596.63  1215.5  569.64
  1742.4  511.39  1940.3  508.98  2072.4  529.77  2458.6  495.42  2741.9  492.67
  2827.4  480.36  3202.1  476.46    3534  485.02 3623.53   452.1    3673     441
  3708.4  446.48    3753  437.93 3848.07   452.4    3861   465.1  3984.8  478.49
  4007.3     495  4063.3  506.07  4092.4  528.54  4180.2  544.69  4266.8  603.87
  4322.2  623.64  4703.6  634.18  5330.6  776.97  5416.2  783.17  5508.3   777.1
#Mann= 3 , 0 , 0
       0      .1       0 3623.53    .035       0 3848.07      .1       0
Bank Sta=3623.53,3848.07
XS Rating Curve= 0 ,0
Exp/Cntr=0.3,0.1

Type RM Length L Ch R = 1 ,26534.84,1373.8,1455.3,1532.5
XS GIS Cut Line= 6
      1990864.89       687311.28      1991082.07       686896.25
      1991442.87       686429.461991781.07911924685404.495151662
1992042.22617782684449.240145402      1993156.19       682564.79
#Sta/Elev= 30
       0  586.93   280.8  602.32   485.4   605.4   691.5  595.71   984.6  594.66
  1323.4  568.15  1771.3  520.14  1952.6  509.36    2457  491.11    2917  486.56
  3197.7  472.58 3360.25  444.54  3449.2  445.89  3537.5  473.93  3614.6  489.13
  3670.8  527.39  3790.3  585.27  3800.5   605.6  3816.5  662.52  3826.7  681.05
  3872.8  734.09  3924.7  769.14  4057.3  826.23  4100.5  854.18    4285  890.41
    4360  891.94  4567.5  844.76    5046   686.8  5152.6  714.91  5317.6  723.12
#Mann= 3 , 0 , 0
       0      .1       0  3197.7    .035       0  3537.5      .1       0
Bank Sta=3197.7,3537.5
XS Rating Curve= 0 ,0
Exp/Cntr=0.3,0.1

Type RM Length L Ch R = 1 ,25079.58,1665.1,1674.1,1706.5
BEGIN DESCRIPTION:
7819.111
END DESCRIPTION:
XS GIS Cut Line= 6
      1990886.55       687465.44      1991167.36       686830.62
      1992176.82       685846.29      1993336.92       685196.02
      1995561.08       683154.27      1998472.23        682808.6
#Sta/Elev= 30
       0  569.59   672.5  599.71  1095.6  587.32  1987.2  535.73  2418.7   478.9
  2994.6   465.4  3169.4  439.87 3266.69  444.19  3312.9   467.9  3347.1  476.59
  3461.5  575.96  3478.3  621.81  3516.9  667.76  3592.3   700.4    4415  653.52
  4685.8  598.25    5022  668.48  5460.2  797.38  6115.2  876.97  6390.1  942.16
  6453.9  942.99  6950.3  805.28  7204.6  781.95    7766  918.31  8096.1  822.41
  8448.3  755.28  8596.8  695.32  8652.2   694.4  9168.3  844.18  9385.5  795.52
#Mann= 3 , 0 , 0
       0      .1       0  2994.6    .035       0  3312.9      .1       0
#XS Ineff= 2 , 0
         2577.59  480.64
Permanent Ineff=
       F       F
Bank Sta=2994.6,3312.9
XS Rating Curve= 0 ,0
Exp/Cntr=0.3,0.1

Type RM Length L Ch R = 1 ,23405.49,1621.7,1622.4,1644.9
XS GIS Cut Line= 6
      1991529.53       688488.64      1992381.92       687610.26
1994345.14271002686592.827955558       1994948.3       686418.69
      1996657.53       685571.01       1999397.9       684987.02
#Sta/Elev= 30
       0  574.45   486.7  530.69    1060  520.85  1213.2  506.61  1552.2  513.23
  1720.3  548.36  1924.9  559.82  2213.1  498.05  2729.4   484.9  2766.3  462.53
 2823.02  442.08 2894.45  440.57 2934.03  441.01  2980.5  462.53  3757.5  493.03
  4015.1  583.62  4114.1  566.02  5586.3  566.36  6245.8  664.65  6389.9   651.5
  6694.8  577.73  6828.3  569.28    7257  667.79  7485.5  677.95  7762.8  640.35
  7983.6  703.63    8171  725.45  8386.8  710.48  8692.6   632.1    8786  631.49
#Mann= 3 , 0 , 0
       0      .1       0  2766.3    .035       0  2980.5      .1       0
Bank Sta=2766.3,2980.5
XS Rating Curve= 0 ,0
Exp/Cntr=0.3,0.1

Type RM Length L Ch R = 1 ,21783.08,1900.4,1938.8,2022.6
BEGIN DESCRIPTION:
6797.347
END DESCRIPTION:
XS GIS Cut Line= 6
      1992173.48       689511.66      1993159.08       688816.59
 1995114.4886029688050.853500289      1995862.71       688281.61
      1998316.82       687898.74      2000323.75       687165.99
#Sta/Elev= 30
       0  859.28     757  691.51  1045.4  586.77  1521.2  495.89  2107.6   489.4
  2338.6   462.7  2431.5  484.17  2609.2  484.35 2668.61  457.02  2785.7  440.55
 2928.02  457.32  3307.2  493.67  3443.2  474.15  4018.7  568.63  4236.2  570.05
  4491.8  546.06  4765.3  612.62  5066.1   714.7  5436.8  816.75  5684.1  862.41
  6118.7  908.21  6374.3     981  6533.7 1007.93  6751.9  990.17  6873.2  959.69
  7119.7  865.18  7673.3  776.45  8099.1  901.31  8514.3  881.11  8710.9  898.71
#Mann= 3 , 0 , 0
       0      .1       0 2668.61    .035       0 2928.02      .1       0
Bank Sta=2668.61,2928.02
XS Rating Curve= 0 ,0
Exp/Cntr=0.3,0.1

Type RM Length L Ch R = 1 ,19844.27,1849.7,1856.7,1875.8
XS GIS Cut Line= 6
      1992415.39       691318.78      1993600.33       690421.52
1995743.57058744689984.861323671      1996088.64        690071.6
      1997088.67       689986.19      1999522.36        687821.2
#Sta/Elev= 30
       0  555.67    85.6  524.59   231.9  571.61   519.9   610.2   682.3  602.29
   924.6  562.69  1102.2  596.66  1243.9  604.61  1614.8  565.98  1678.7  551.33
  1811.5   490.6  1870.2  484.92  3081.3   482.4  3181.6  459.77 3243.79  441.37
  3467.9  461.81  3498.4  480.43  3635.2   496.5  3965.2  499.78  4300.7  536.21
  4980.6  508.33  5695.4  612.65  6246.8  616.92  6590.2  656.37  6838.8  723.93
  7122.4  831.13  7393.7  882.55  7530.8  829.42    7766  784.33  8296.4     776
#Mann= 3 , 0 , 0
       0      .1       0  3181.6    .035       0  3467.9      .1       0
#XS Ineff= 2 , 0
         2572.76  487.51
Permanent Ineff=
       F       F
Bank Sta=3181.6,3467.9
XS Rating Curve= 0 ,0
Exp/Cntr=0.5,0.3

Type RM Length L Ch R = 1 ,17987.56,186.9,187.2,186.5
BEGIN DESCRIPTION:
5611.002
END DESCRIPTION:
XS GIS Cut Line= 5
       1992657.3       693125.891993880.59813086692023.670682225
       1995764.3       691870.491997292.27356074691787.986330207
  1998590.503421688757.649514727
#Sta/Elev= 30
       0   580.1     195  597.61   478.8  600.94   751.5  586.66   949.4   595.5
  1393.8  558.28  1838.2  535.68  1998.7  506.21  2099.1  504.09  2139.2  523.63
  2170.2  523.73  2284.7  489.76  2540.5  473.91  2886.7  468.75  2990.4  442.23
  3157.3  445.13 3261.68472.4565  3380.5  487.95  3876.8  486.32  4107.1  491.62
  4154.7  500.04  4217.3  491.94  4420.1  493.62    5075  521.99  5469.4  507.13
  6734.1  538.07  7528.3  591.19  7887.2  629.02  8239.2  729.12  8363.5  773.03
#Mann= 3 , 0 , 0
       0      .1       0  2886.7    .035       0 3261.68      .1       0
Bank Sta=2886.7,3261.68
XS Rating Curve= 0 ,0
Exp/Cntr=0.5,0.3

Type RM Length L Ch R = 3 ,17899.2 ,,,
BEGIN DESCRIPTION:
Cookeville Hwy
2019 Update:
-Removed tressle as this is open space.
END DESCRIPTION:
Bridge Culvert--1,0,-1,-1, 0
Deck Dist Width WeirC Skew NumUp NumDn MinLoCord MaxHiCord MaxSubmerge Is_Ogee
77,50,2.61,0, 35, 35, , , 0.95, 0, 0,0,,
    1825 2358.25 2478.152478.151 2479.84 2522.13 2565.04 2608.01 2651.05 2694.04
 2737.04 2779.82 2822.92 2865.51  2907.8 3025.29 3070.73  3255.3 3369.15 3414.01
 3456.91 3499.33 3527.37 3556.11 3584.75 3612.97 3641.48 3669.92 3698.52 3726.73
 3756.65 3756.66 3756.67 3992.86 5200.19
  546.89  514.71  513.27  513.27  512.76  512.66  512.87   513.7  515.14  516.88
  518.64  520.36  522.08  523.82  529.81   536.2   536.2  533.81  528.84  524.62
  523.21  522.32  520.02  518.84  517.77   516.6  515.48  514.32  513.15  511.91
  510.77  510.77  507.67  503.25  522.26
                          506.67  506.67  506.06  506.27   507.1  508.54  510.28
  512.04  513.76  515.48  517.22  519.06  525.45  525.45  523.06  518.09  518.01
  516.21  515.67  514.01  513.33  512.16  511.05  509.93  508.77   507.6  506.36
  504.87
    1668 2201.25 2321.152321.151 2322.84 2365.23 2408.08 2450.85 2494.08 2536.98
 2580.03 2623.06 2665.93 2708.85 2751.06 2868.29 2913.73 3098.85 3212.44 3255.89
 3298.88 3341.97 3370.47 3398.63 3426.99 3455.98 3484.31 3513.01  3541.7 3570.26
 3599.89  3599.9 3599.91 3835.86 5667.19
  546.89  514.71  513.27  513.27  512.76  512.67  512.89  513.69  515.15  516.93
  518.68  520.39  522.08  523.77  529.81   536.2   536.2  533.81  528.95  523.89
  522.57   521.2  521.12  518.84   518.3   516.6   515.5  514.29  513.12  512.03
   510.8   510.8  507.67  503.25     521
                          506.67  506.67  506.07  506.29  507.09  508.55  510.33
  512.08  513.79  515.47  517.17  519.07  525.45  525.45  523.03  518.09  517.29
  515.57  514.55  514.52  513.33   512.2  511.05  509.95  508.74  507.57  506.48
  504.87
Pier Skew, UpSta & Num, DnSta & Num=  ,2522.13, 2 ,2365.23, 2 , 2 , 2 , 0 ,,
     2.5       3
   491.5  505.57
     2.5       3
   491.5  505.57
Pier Skew, UpSta & Num, DnSta & Num=  ,2565.04, 2 ,2408.08, 2 , 2 , 2 , 0 ,,
     2.5       3
  484.95  505.79
     2.5       3
  484.95  505.79
Pier Skew, UpSta & Num, DnSta & Num=  ,2607.85, 2 ,2451.01, 2 , 2 , 2 , 0 ,,
     2.5       3
  482.41  506.59
     2.5       3
  482.41  506.59
Pier Skew, UpSta & Num, DnSta & Num=  ,2651.05, 2 ,2494.08, 2 , 2 , 2 , 0 ,,
       2       3
  481.17  508.04
       2       3
  481.17  508.04
Pier Skew, UpSta & Num, DnSta & Num=  ,2694.04, 2 ,2536.98, 2 , 2 , 2 , 0 ,,
       2       3
  480.34  509.78
       2       3
  480.34  509.78
Pier Skew, UpSta & Num, DnSta & Num=  ,2737.04, 2 ,2580.03, 2 , 2 , 2 , 0 ,,
       2       3
  478.48  511.58
       2       3
  478.48  511.58
Pier Skew, UpSta & Num, DnSta & Num=  ,2780.06, 2 ,2622.82, 2 , 2 , 2 , 0 ,,
       2       3
  475.71  513.26
       2       3
  475.71  513.26
Pier Skew, UpSta & Num, DnSta & Num=  ,2822.92, 2 ,2665.93, 2 , 2 , 2 , 0 ,,
       2       3
  474.11  514.97
       2       3
  474.11  514.97
Pier Skew, UpSta & Num, DnSta & Num=  ,2865.51, 2 ,2708.85, 2 , 2 , 2 , 0 ,,
       2       3
  473.78  516.67
       2       3
  473.78  516.67
Pier Skew, UpSta & Num, DnSta & Num=  ,2909.22, 3 ,2751.8, 3 , 0 , 0 , 0 ,,
    3.42    3.42       2
  474.46  518.47  520.33
    3.42    3.42       2
  474.46  518.47  520.33
Pier Skew, UpSta & Num, DnSta & Num=  ,3369.44, 3 ,3212.15, 3 , 0 , 0 , 0 ,,
    3.27    3.27       2
  476.95  518.98  521.84
    3.27    3.27       2
  476.95  519.01  521.95
Pier Skew, UpSta & Num, DnSta & Num=  ,3414.01, 2 ,3255.89, 2 , 2 , 2 , 0 ,,
       2       3
  481.16  517.51
       2       3
  481.16  516.79
Pier Skew, UpSta & Num, DnSta & Num=  ,3456.91, 2 ,3298.88, 2 , 2 , 2 , 0 ,,
       2       3
  487.97  515.71
       2       3
  487.97  515.07
Pier Skew, UpSta & Num, DnSta & Num=  ,3499.33, 2 ,3341.97, 2 , 2 , 2 , 0 ,,
       2       3
  491.03  515.17
       2       3
  491.03  515.17
Pier Skew, UpSta & Num, DnSta & Num=  ,3527.37, 2 ,3370.47, 2 , 2 , 2 , 0 ,,
       2       3
  490.88  514.01
       2       3
  490.88  514.02
Pier Skew, UpSta & Num, DnSta & Num=  ,3555.63, 2 ,3399.11, 2 , 2 , 2 , 0 ,,
       2       3
  490.43  512.83
       2       3
  490.43  512.83
Pier Skew, UpSta & Num, DnSta & Num=  ,3584.75, 2 ,3426.99, 2 , 2 , 2 , 0 ,,
       2       3
  490.64  511.66
       2       3
  490.64   511.7
Pier Skew, UpSta & Num, DnSta & Num=  ,3612.97, 2 ,3455.98, 2 , 2 , 2 , 0 ,,
       2       3
  491.05  510.55
       2       3
  491.05  510.55
Pier Skew, UpSta & Num, DnSta & Num=  ,3641.48, 2 ,3484.31, 2 , 2 , 2 , 0 ,,
       2       3
  490.54  509.43
       2       3
  490.54  509.45
Pier Skew, UpSta & Num, DnSta & Num=  ,3670.01, 2 ,3512.92, 2 , 2 , 2 , 0 ,,
       2       3
  490.27  508.24
       2       3
  490.27  508.27
Pier Skew, UpSta & Num, DnSta & Num=  ,3698.52, 2 ,3541.7, 2 , 2 , 2 , 0 ,,
       2       3
  489.82   507.1
       2       3
  489.82  507.07
Pier Skew, UpSta & Num, DnSta & Num=  ,3726.73, 2 ,3570.26, 2 , 2 , 2 , 0 ,,
     2.5       3
  489.45  505.86
     2.5       3
  489.45  505.68
BR Coef=-1 , 1 , 0 ,, 0 ,,,0.8,0,1.33,0,
WSPro=,,,, 1 ,,,, 0 ,,,, 0 ,,,,-1 ,-1 ,-1 , 0 , 0 , 0 , 0 , 0
BC Design=,, 0 ,, 0 ,,,,,,
BC HTab HWMax=600
BC Use User HTab Curves=0
BC User HTab FreeFlow(D)= 0

Type RM Length L Ch R = 1 ,17800.40,451.9,481.9,505.7
XS GIS Cut Line= 5
1992689.66657572693156.5951667011993782.95683978692212.239768405
1995656.31051694692065.4817999741997337.89266705691943.355722033
1998798.08853691688588.876682762
#Sta/Elev= 30
       0  582.59   180.9  599.09     457  607.26   766.8     595   973.7  599.62
  1347.5  574.58  1454.4     559  2288.4  510.56  2411.2  483.09  2759.7 469.402
    2810  464.72  2869.4442.1654  3036.3445.0654  3128.4  470.39  3398.9  491.21
  4409.4  493.06  5009.8  525.55  5056.7  524.89  5075.7  515.67  5233.9  523.88
  5515.4  510.45  6002.7  530.14  6863.2  543.44  7292.5  573.82  7520.5  599.59
  7701.4  606.94  7998.6  641.33  8039.5  637.66  8549.4  809.62  8668.3   836.1
#Mann= 3 , 0 , 0
       0      .1       0  2759.7    .035       0  3128.4      .1       0
Bank Sta=2759.7,3128.4
XS Rating Curve= 0 ,0
Exp/Cntr(USF)=0,0
Exp/Cntr=0.5,0.3

Type RM Length L Ch R = 1 ,17318.46,2074.7,1947.1,1801.4
BEGIN DESCRIPTION:
5451.291
END DESCRIPTION:
XS GIS Cut Line= 6
      1993667.76       692663.28      1994252.47       692768.04
1994741.59985877692541.607793933      1996348.09       692586.63
      1996854.54       692756.28      1999117.35       688669.28
#Sta/Elev= 30
       0  595.68   224.8  583.54   537.1  586.45   775.5  568.73     903  577.51
  1092.2  531.94  1203.2  484.21  1481.1   464.1 1538.17  441.69 1570.42  441.39
 1720.88  442.74  1803.8  465.01  1910.2     478  2229.9  492.54  2517.6  479.94
  2718.1  487.79  2993.3  480.88  3449.4   499.6  3774.6  484.63  4133.4   525.5
  4335.1   528.6  4356.6  516.46  4486.2  523.29  4758.9  513.24  5206.7  541.99
  5709.8  542.89  6527.2  607.86  6839.3  646.57  7637.7   766.7  7953.8  786.81
#Mann= 3 , 0 , 0
       0      .1       0  1481.1    .045       0  1803.8      .1       0
#XS Ineff= 2 , 0
                         2231.01          492.54
Permanent Ineff=
       F       F
Bank Sta=1481.1,1803.8
XS Rating Curve= 0 ,0
Exp/Cntr=0.3,0.1

Type RM Length L Ch R = 1 ,15371.36,1487,1676.2,1770.9
XS GIS Cut Line= 6
1994445.59647476694277.2105808861995631.25529237694474.360580886
      1996093.61       694192.02      1996542.66       694280.95
      1998197.18       693415.052003889.22207685692723.906209724
#Sta/Elev= 30
       0  549.37   187.2  549.86     395  532.31   651.3  551.83    1197  511.16
  1304.6  491.07 1398.09455.0192 1495.31  438.71 1640.11  455.12    1782  478.36
  1994.9  463.07  2182.5  481.86    3627  463.86  4304.7  475.22    4758  510.16
  5062.7  604.47    5234  644.73  5606.7   672.1    5924   660.2  6246.5  594.71
  6644.3  549.11  6980.8  493.43  7213.4  488.15  7374.6  509.87  7943.7  532.46
  8487.4  630.95  8817.4  610.06  9321.3  710.08  9603.3  787.77  9847.8  836.92
#Mann= 3 , 0 , 0
       0      .1       0 1398.09     .04       0 1640.11      .1       0
#XS Ineff= 1 ,-1
 2360.74  4847.3     483
Permanent Ineff=
       F
Bank Sta=1398.09,1640.11
XS Rating Curve= 0 ,0
Exp/Cntr=0.3,0.1

Type RM Length L Ch R = 1 ,13695.17,1335.3,1607.2,1803.5
BEGIN DESCRIPTION:
4262.708
END DESCRIPTION:
XS GIS Cut Line= 6
       1994393.6       694343.78      1994787.37       694805.11
      1995873.12       695829.451997029.06117208695707.059412674
      1998141.69       696480.43      1998697.31       697792.71
#Sta/Elev= 30
       0  558.19   317.6  552.93     615  517.96   761.8  520.08     898  539.88
  1271.1  539.76  1455.8  526.16  1759.2  485.27  1976.8  497.41  2274.3   493.3
  2457.2  484.83  2542.6  461.81  2778.9  465.34 2902.79  456.71  3015.2  436.02
 3111.58  461.72    3181  477.13  3231.5  501.27  3289.4  536.08  3321.4  577.94
  3344.2  596.02    3549   584.4  3632.7  564.11  3669.9  575.32  3812.5  584.37
  4178.5  584.21  4968.6  712.05  5183.1  732.07  5375.8  727.93  6043.5  684.88
#Mann= 3 , 0 , 0
       0      .1       0 2902.79    .035       0 3111.58      .1       0
Bank Sta=2902.79,3111.58
XS Rating Curve= 0 ,0
Exp/Cntr=0.3,0.1

Type RM Length L Ch R = 1 ,12088.00,819.9,971.7,1097.5
XS GIS Cut Line= 6
      1994352.28       694364.59      1995235.61       695687.64
      1995405.11       696385.351995910.27529238697112.131763266
      1996791.77       698244.97      1997435.93       699769.14
#Sta/Elev= 30
       0  562.21   165.9  551.91   625.8  536.92   755.8  526.76  1007.1  535.76
  1278.1  534.98    1818  490.84  2188.5  492.06  2525.5  482.04  2707.4  481.58
  2828.8  462.61 2875.57  448.82 2982.79  444.51 3035.16  446.62  3161.9  463.51
  3186.2   465.2  3216.4  482.78    3244   490.6  3396.7  505.07  3705.1  514.73
  4027.3  507.22  4095.3  510.59  4200.6  506.38  4283.1  510.94  4447.7  508.42
  4685.6  535.45  5415.7  559.45  5803.8   564.9  6189.2  588.49  6288.3  589.41
#Mann= 3 , 0 , 0
       0      .1       0  2828.8    .035       0  3161.9      .1       0
Bank Sta=2828.8,3161.9
XS Rating Curve= 0 ,0
Exp/Cntr=0.3,0.1

Type RM Length L Ch R = 1 ,11116.30,636.7,647,661.9
BEGIN DESCRIPTION:
3432.218
END DESCRIPTION:
XS GIS Cut Line= 6
      1994310.65       694386.32      1994523.65        694828.7
      1994828.83       695457.67      1995112.63       696031.33
      1994691.09       698227.411995685.94891032700572.606112642
#Sta/Elev= 30
       0  559.73   779.1  523.88  1013.1  535.04  1343.7  530.86  1650.5  495.62
  1817.9  486.31  2807.3  481.61 2890.91  453.37  3029.1  433.83 3116.21  441.36
 3141.37  454.02  3172.8  462.57  3178.3  500.93  3184.2     529  3201.2  568.71
  3247.1  614.73    3410  610.94    3731  669.93  4032.1  745.33  4131.5  760.21
  4224.3  759.94  4375.9  739.47  5112.3  590.52  5196.5  591.76  5343.1  617.58
  5597.5  686.07  5989.5  754.58    6280  768.77  6358.9  764.16  6613.8  791.41
#Mann= 3 , 0 , 0
       0      .1       0 2890.91    .035       0 3141.37      .1       0
#XS Ineff= 2 , 0
         2748.06   481.9
Permanent Ineff=
       F       F
Bank Sta=2890.91,3141.37
XS Rating Curve= 0 ,0
Exp/Cntr=0.3,0.1

Type RM Length L Ch R = 1 ,10469.31,802.2,848.8,901
XS GIS Cut Line= 6
       1994280.9       694352.07      1994429.69       694800.88
      1994701.28       695683.26      1994298.66       696902.53
      1994156.39        697438.3      1994968.49        700409.5
#Sta/Elev= 30
       0  556.07     110  558.58   340.5  531.44   818.6  517.54  1296.2  538.09
    1477  526.45  1732.6  488.31  1995.8  499.35  2619.9  479.71  2688.2  461.31
 2738.23  440.71 2796.78   434.6 2873.73   438.8  2957.2  461.31  3003.8  495.66
  3009.1   531.3  3011.6  562.41  3021.9  581.03  3045.2  592.19  3363.6  578.23
  3550.3  601.68  4249.2  762.77  4356.6   761.4  4911.4  680.37  5225.1  621.13
  5318.3  617.07  5390.9  626.83  6064.3   804.1  6206.8  855.63  6314.6  876.45
#Mann= 3 , 0 , 0
       0      .1       0  2688.2    .035       0  2957.2      .1       0
#XS Ineff= 2 , 0
         2573.31  479.94
Permanent Ineff=
       F       F
Bank Sta=2688.2,2957.2
XS Rating Curve= 0 ,0
Exp/Cntr=0.3,0.1

Type RM Length L Ch R = 1 ,9620.471,810.7,837,857.8
XS GIS Cut Line= 6
      1994251.77       694317.23      1994295.88       694689.23
      1994290.32       695335.35      1993783.13        696214.8
1993387.08706208696844.3617619781992693.51707367697784.461782587
#Sta/Elev= 30
       0  549.89   144.6   559.1   199.5  548.16   227.9   558.1   470.8  520.28
   770.6  506.41   951.7  523.65  1068.5  525.94  1468.3  492.68  1776.9  491.45
  1836.2  477.97  1918.6  477.64  1984.7  488.38  2148.9   476.8  2296.6  480.75
    2397  467.73 2429.68  457.28 2567.45  435.38 2654.05  438.78    2715  461.31
    2840  492.85  2855.6  504.96  2860.6  531.68  2864.8  543.13    2872  574.35
  2879.2  584.37  2970.4  599.74  3038.9  622.78  3408.4  688.37    3948  721.28
#Mann= 3 , 0 , 0
       0      .1       0 2429.68    .035       0    2715      .1       0
Bank Sta=2429.68,2715
XS Rating Curve= 0 ,0
Exp/Cntr=0.3,0.1

Type RM Length L Ch R = 1 ,8783.463,929,934.9,939.5
XS GIS Cut Line= 6
      1994222.65       694282.39      1994161.06       694577.68
      1993879.27       694986.46       1993267.6       695527.06
1992654.64411901696381.425303967      1992557.16       697733.62
#Sta/Elev= 30
       0  548.85   197.1   563.1   235.4  556.25     266  542.48   375.5  549.97
   708.8  519.57   929.3  524.69  1265.9  490.45  1369.6  491.41  1641.6  478.22
  2133.8  478.44  2227.9  466.49 2329.58  438.86 2378.12  436.15 2474.38  438.75
 2510.53  448.33  2526.3  461.16  2594.5  474.33    2640  498.78  2650.6  539.31
  2655.9  544.82  2849.9  549.96  2957.7  533.09  3000.3  550.47  3155.7  572.44
  3363.7  614.59  3621.9  690.48  3824.9  737.93  3910.1  751.91  4026.2  756.24
#Mann= 3 , 0 , 0
       0      .1       0  2227.9    .035       0  2526.3      .1       0
Bank Sta=2227.9,2526.3
XS Rating Curve= 0 ,0
Exp/Cntr=0.3,0.1

Type RM Length L Ch R = 1 ,7848.611,625.7,671.1,706.3
BEGIN DESCRIPTION:
2412.344
END DESCRIPTION:
XS GIS Cut Line= 6
      1994192.63       694248.64      1994026.25       694466.14
       1993424.1       694652.09      1992752.17       694840.31
      1991784.38       695947.82      1991351.55       696396.16
#Sta/Elev= 30
       0  552.13   172.2  559.62   370.3   553.1   490.7  538.38   590.1   533.5
     666  536.75   710.8  528.07   754.9  529.85  1210.4  492.48  1388.9     483
  1555.8  487.12  1655.5  477.91  1982.7  481.88  2179.6  475.25  2345.6  479.99
  2438.6  465.91 2469.47  456.32  2522.8  438.32  2568.8  436.92  2674.7  438.72
 2754.33   458.2  2810.7  484.67  2895.7  480.58  3046.1  484.15  3148.9  494.71
  3329.3  524.99  3348.7  531.91  3375.4   531.5  3562.6   585.4  3695.8  614.44
#Mann= 3 , 0 , 0
       0      .1       0 2469.47    .035       0 2754.33      .1       0
Bank Sta=2469.47,2754.33
XS Rating Curve= 0 ,0
Exp/Cntr=0.3,0.1

Type RM Length L Ch R = 1 ,7177.535,439.7,451,461.1
XS GIS Cut Line= 6
      1993486.91       693708.14      1993273.09       693937.52
      1992550.49       694258.511992197.13117465694692.552940495
1991225.03882921695420.005297527      1991210.24       696554.27
#Sta/Elev= 30
       0  530.52   163.7  527.66   304.8  508.47   394.2  522.61   443.9  523.72
   983.2  517.51  1113.9  511.26    1271  493.81  1330.9  472.89  1422.3  472.88
  1565.1  482.75  1683.5  481.99  1828.4  472.92  2076.6   478.5  2135.8  476.85
 2256.86  459.37 2321.38  438.32 2337.47  440.24 2365.05   434.8 2459.81  437.77
  2543.9  461.03  2583.4   482.9  2898.9  477.06    3054  482.05  3349.2  524.12
    3539  565.73    3684  603.86    3849  638.37    3944  646.18  4012.9     643
#Mann= 3 , 0 , 0
       0      .1       0 2256.86    .035       0  2543.9      .1       0
#XS Ineff= 2 , 0
          1574.5  482.77 2583.69          482.93
Permanent Ineff=
       F       F
Bank Sta=2256.86,2543.9
XS Rating Curve= 0 ,0
Exp/Cntr=0.3,0.1

Type RM Length L Ch R = 1 ,6726.529,699.5,706.2,713.7
XS GIS Cut Line= 5
       1992781.3       693168.621991992.43999742694322.442934054
1990975.09353297695012.8276532721990990.75823931695355.687650696
      1991068.93       696712.37
#Sta/Elev= 30
       0  596.72   288.9  596.79   538.2  566.04   865.2   568.6  1134.8  531.99
  1173.4   504.2  1249.9  472.11  1331.6  472.27  1346.8  479.63  1391.5  481.76
  1573.2  471.89  1861.2  477.05  1972.8  473.03    2044  461.17 2073.18  449.59
 2133.89  438.43 2156.21  441.21  2176.3  432.67  2329.8  448.77  2355.7  464.54
  2395.8  483.78  2922.6  476.38  3002.7  479.41  3137.9  509.84  3248.1  514.61
  3348.2  504.27  3636.4   564.1  4019.3  664.29    4122  674.69  4329.3  671.84
#Mann= 3 , 0 , 0
       0      .1       0    2044    .035       0  2355.7      .1       0
#XS Ineff= 2 , 0
          1414.8  481.91 2396.29          483.78
Permanent Ineff=
       F       F
Bank Sta=2044,2355.7
XS Rating Curve= 0 ,0
Exp/Cntr=0.3,0.1

Type RM Length L Ch R = 1 ,6020.35 ,1364.9,1191.2,1030.3
XS GIS Cut Line= 5
       1992076.7         692629.1991478.89999227693846.251170788
1990399.63861609694521.8585313051990197.74471278694953.528813755
      1990927.61       696870.48
#Sta/Elev= 30
       0  587.55   116.9  593.32   594.8  564.13   849.2  566.53   970.6  547.91
  1024.7  548.13  1135.1  566.84    1275  573.24  1313.4  562.95  1355.2  501.65
  1433.4  474.54  1730.9  473.09 1775.55  462.79 1864.83  445.12 1965.05  442.77
 1984.55  430.55 2125.19  445.41  2146.2  462.05  2230.8  480.26  2627.1  480.91
  2882.6  469.76  3196.2  482.51  3329.3  499.77  3701.8  500.22  3815.6  519.31
  4022.9  530.72  4295.7  571.74  4900.2  715.34  5020.6  729.51  5157.2  726.56
#Mann= 3 , 0 , 0
       0      .1       0 1775.55    .035       0  2146.2      .1       0
#XS Ineff= 2 , 0
                         2307.35          481.41
Permanent Ineff=
       F       F
Bank Sta=1775.55,2146.2
XS Rating Curve= 0 ,0
Exp/Cntr=0.3,0.1

Type RM Length L Ch R = 1 ,4829.109,1482.6,1480.1,1475.5
BEGIN DESCRIPTION:
1470.010
END DESCRIPTION:
XS GIS Cut Line= 6
      1991370.98       692088.491990080.58058861693228.257644255
 1990039.5503858693943.5350099251989811.87882277694619.951178516
1990072.30764426695068.257056929       1990786.3       697028.59
#Sta/Elev= 30
       0  604.17   133.8  596.18   589.6  592.03  1183.3  568.89  1486.9  541.78
  1761.4  533.08  1799.4  524.08  1811.5  512.09  1821.5  488.04 1862.54  462.88
  1942.9  438.63  1963.9  444.33  1981.7  428.53  2049.9  435.63  2056.5  447.73
  2091.9  463.09  2186.9  478.25  2651.3  480.37  2858.4  476.36  2962.4  465.93
  3151.8  476.86    3589   480.5  3604.1  486.67  3733.8  491.25  4356.4  501.01
  4734.7   553.9  5050.8  627.58    5394  726.46  5554.1  760.77  5756.6  781.09
#Mann= 3 , 0 , 0
       0      .1       0 1862.54    .035       0  2091.9      .1       0
#XS Ineff= 2 , 0
                         2575.32          480.72
Permanent Ineff=
       F       F
Bank Sta=1862.54,2091.9
XS Rating Curve= 0 ,0
Exp/Cntr=0.3,0.1

Type RM Length L Ch R = 1 ,3349.039,1338,1334.1,1330.6
XS GIS Cut Line= 5
 1988889.1356792691580.3767313531988609.09169042692941.873268647
1988562.39319967694085.412285477      1989097.64       694673.27
       1990533.7       696728.02
#Sta/Elev= 30
       0  883.55   336.9  793.17   660.5  694.35  1028.6   610.8  1181.3  586.36
  1301.7  552.59  1365.5  515.51  1463.6  499.26  1498.6  501.34  1546.1  483.25
 1694.58  448.88 1768.72  438.61 1780.93  443.74 1813.83  430.33 1958.27  444.91
  2009.3  463.16  2109.1  477.93  2301.4  474.14  2669.7  488.21  2842.1  482.65
  2986.3  491.09  3353.4  489.81  4021.4  520.38  4384.4  506.81    4657  514.17
  4832.7  511.26  5032.2  528.34  5314.1   573.5  5512.9  623.79  5836.4  717.59
#Mann= 3 , 0 , 0
       0      .1       0 1694.58    .035       0 1958.27      .1       0
#XS Ineff= 2 , 0
                         2141.58          477.97
Permanent Ineff=
       F       F
Bank Sta=1694.58,1958.27
XS Rating Curve= 0 ,0
Exp/Cntr=0.3,0.1

Type RM Length L Ch R = 1 ,2014.892,1355.7,1149.2,965.6
XS GIS Cut Line= 5
1987309.77962662691249.6856609461987249.51372168693678.712486929
1987647.86793873694184.0249215721989849.61663407695897.717617642
1990520.49003137696882.987872301
#Sta/Elev= 30
       0  815.63   220.5  770.31   640.9  707.84  1201.1  571.06  1501.2  526.05
  1591.2   521.2  1633.7  494.13  1656.2  487.54  1716.2  481.87  1771.2  485.36
  1896.3   462.8 1977.06  439.25 1999.35  441.43 2035.87  432.24 2142.18  439.71
 2200.84  455.02  2278.9  463.92  2353.9  482.03  2673.8  473.19  2998.5  482.41
  3221.1   475.5  3535.4  476.89  4687.3  493.94  5029.1  514.87  5411.8  496.89
  5741.4  518.95  5973.4  518.07  6248.1   546.3    6446  579.87  7055.3  749.31
#Mann= 3 , 0 , 0
       0      .1       0  1896.3    .035       0  2278.9      .1       0
#XS Ineff= 2 , 0
                         2354.15          482.03
Permanent Ineff=
       F       F
Bank Sta=1896.3,2278.9
XS Rating Curve= 0 ,0
Exp/Cntr=0.3,0.1

Type RM Length L Ch R = 1 ,865.689 ,0,0,0
BEGIN DESCRIPTION:
173.0832
END DESCRIPTION:
XS GIS Cut Line= 6
      1984141.05       693805.351985937.95991114693377.134119011
1986350.29012981693742.4420969811987457.01629575694235.903808821
1989575.14405309696072.9140171921990545.09038014697023.607617642
#Sta/Elev= 30
       0  694.41   288.4  688.63   506.9  652.39   532.5  628.34   553.1  589.88
   571.1   583.5   591.6  556.26   753.5  556.97   763.8  576.86   799.8   585.7
   838.4  622.73    1414  538.98  1550.2  542.63  1640.2  523.73  1778.9   461.5
  1892.1  462.64    1959  438.74  2023.9  434.14  2272.9  460.46  2623.6  482.94
  3131.1  474.36  5926.3  485.17  6068.6   502.4  6244.6   550.8  6352.1   564.5
  6492.2  571.73  6727.4  558.83  6925.6  575.87  7220.8  632.92    7779  772.07
#Mann= 3 , 0 , 0
       0      .1       0  1892.1    .035       0  2272.9      .1       0
Bank Sta=1892.1,2272.9
XS Rating Curve= 0 ,0
Exp/Cntr=0.3,0.1
Stream Node=Caney Fork      ,Reach - 1       , 0 , 0 ,Upstream end
Stream Node=Caney Fork      ,Reach - 1       , 0 , 1 ,Downstream end
LCMann Table=0

Chan Stop Cuts=-1
Use User Specified Reach Order=0
Composite Channel Slope=5
