--- SmithFork2019.prj (project) ---

Proj Title=Smith County FPMS Study 2019
Current Plan=p01
Default Exp/Contr=0.3,0.1
English Units
Geom File=g07
Geom File=g02
Flow File=f04
Flow File=f06
Plan File=p01
Background Map Layer=Google Map
Background Map Layer=Google Satellite
Y Axis Title=Elevation
X Axis Title(PF)=Main Channel Distance
X Axis Title(XS)=Station
BEGIN DESCRIPTION:
Smith Fork River
END DESCRIPTION:
DSS File=dss
DSS Export Rating Curves= 0
DSS Export Rating Curve Sorted= 0
DSS Export Volume Flow Curves= 0
DXF Filename=..\Lancaster_HEC-RAS_5_0_3\HEC-RAS_5_0_3\Smith Fork River.
DXF OffsetX= 0
DXF OffsetY= 0
DXF ScaleX= 1
DXF ScaleY= 10

--- SmithFork2019.p01 (plan) ---

Plan Title=2019 Smith Fork 2019 Revision
Program Version=5.07
Short Identifier=2019Revision
Geom File=g07
Flow File=f04
Subcritical Flow
K Sum by GR= 0
Std Step Tol= 0.01
Critical Tol= 0.01
Num of Std Step Trials= 20
Max Error Tol= 0.3
Flow Tol Ratio= 0.001
Split Flow NTrial= 30
Split Flow Tol= 0.02
Split Flow Ratio= 0.02
Log Output Level= 0
Friction Slope Method= 1
Unsteady Friction Slope Method= 2
Unsteady Bridges Friction Slope Method= 1
Parabolic Critical Depth
Global Vel Dist= 0 , 0 , 0
Global Log Level= 0
CheckData=True
Encroach Param=-1 ,0,0, 2
Encroach River=Smith Fork River
Encroach Reach=Reach-1
Encroach Node=26257
       1  1618.8 2420.95
Encroach Node=25342
       1    5100    5972
Encroach Node=24480
       1    4600    5353
Encroach Node=23973
       1  302.67     900
Encroach Node=23424
       1     399    1000
Encroach Node=23044
       1     360    1000
Encroach Node=22489
       1    1008    1800
Encroach Node=21892
       1 1142.46    1950
Encroach Node=21545
       1     930    1750
Encroach Node=20968
       1   875.6    1500
Encroach Node=20370
       1     790    1247
Encroach Node=19864
       1     650 1172.51
Encroach Node=19421
       1     500    1125
Encroach Node=19103
       1     400    1050
Encroach Node=18465
       1     450    1175
Encroach Node=18057
       1     625    1200
Encroach Node=17593
       1     670    1380
Encroach Node=17177
       1     550    1430
Encroach Node=16367
       1     375    1321
Encroach Node=15901
       1     275  1126.1
Encroach Node=15274
       1     175    1025
Encroach Node=14916
       1  240.19    1050
Encroach Node=14500
       1     215     950
Encroach Node=13996
       1   316.9     930
Encroach Node=13527
       1     131     620
Encroach Node=13056
       1     440     890
Encroach Node=11972
       1   504.8    1100
Encroach Node=11529
       1     430     950
Encroach Node=11142
       1     580    1065
Encroach Node=10509
       1     600  1001.3
Encroach Node=10215
       1     475     940
Encroach Node=9984
       1     530    1000
Encroach Node=9677
       1    2430    3200
Encroach Node=9185
       1    5000 5822.59
Encroach Node=8527
       1    4449  5147.8
Encroach Node=7992
       1     198     700
Encroach Node=7500
       1     186     700
Encroach Node=7072
       1     230     700
Encroach Node=6510
       1     250     700
Encroach Node=5841
       1     500    1200
Encroach Node=5085
       1     650  1270.8
Encroach Node=3987
       1  975.76    1607
Encroach Node=2952
       1     550    1140
Encroach Node=2425
       1     700    1300
Encroach Node=2017
       1     600    1300
Encroach Node=1331
       1   225.1     850
Encroach Node=682
       1   105.5     450
Encroach Node=512
       1   172.4     450
Encroach Node=391
       1  185.84   454.1
Encroach Node=350
       1   315.3     730
Computation Interval=1MIN
Output Interval=1HOUR
Instantaneous Interval=1HOUR
Mapping Interval=1HOUR
Computation Time Step Use Courant=        0
Computation Time Step Use Time Series=    0
Computation Time Step Count To Double=0
Computation Time Step Max Doubling=0
Computation Time Step Max Halving=0
Computation Time Step Residence Courant=0
Run HTab= 0
Run UNet= 0
Run Sediment= 0
Run PostProcess= 0
Run WQNet= 0
Run RASMapper= 0
UNET Theta= 1
UNET Theta Warmup= 1
UNET ZTol= 0.02
UNET ZSATol= 0.02
UNET MxIter= 20
UNET Max Iter WO Improvement= 0
UNET MaxInSteps= 0
UNET DtIC= 0
UNET DtMin= 0
UNET MaxCRTS= 20
UNET WFStab= 2
UNET SFStab= 1
UNET WFX= 1
UNET SFX= 1
UNET 1D Methodology=Finite Difference
UNET DSS MLevel= 4
UNET Pardiso=0
UNET DZMax Abort= 100
UNET Use Existing IB Tables=-1
UNET Froude Reduction=False
UNET Froude Limit= 0.8
UNET Froude Power= 4
UNET D1 Cores= 0
UNET D2 Coriolis=0
UNET D2 Cores= 0
UNET D2 Theta= 1
UNET D2 Theta Warmup= 1
UNET D2 Z Tol= 0.01
UNET D2 Volume Tol= 0.01
UNET D2 Max Iterations= 20
UNET D2 Equation= 0
UNET D2 RampUpFraction=0.1
UNET D2 TimeSlices= 1
UNET D2 BCVolumeCheck=0
UNET D1D2 MaxIter= 0
UNET D1D2 ZTol=0.01
UNET D1D2 QTol=0.1
UNET D1D2 MinQTol=1
Write IC File= 0
Write IC File at Fixed DateTime=0
Write IC File at Sim End=0
Echo Input=False
Echo Parameters=False
Echo Output=False
Write Detailed= 0
HDF Write Warmup=0
HDF Write Time Slices=0
HDF Flush=0
HDF Face Node Velocities=0
HDF Compression= 1
HDF Chunk Size= 1
HDF Spatial Parts= 1
HDF Use Max Rows=0
HDF Fixed Rows= 1
Calibration Method= 0
Calibration Iterations= 20
Calibration Max Change=0.05
Calibration Tolerance=0.2
Calibration Maximum=1.5
Calibration Minimum=0.5
Calibration Optimization Method= 1
WQ AD Non Conservative
WQ ULTIMATE=-1
WQ Max Comp Step=1HOUR
WQ Output Interval=15MIN
WQ Output Selected Increments= 0
WQ Output face flow=0
WQ Output face velocity=0
WQ Output face area=0
WQ Output face dispersion=0
WQ Output cell volume=0
WQ Output cell surface area=0
WQ Output cell continuity=0
WQ Output cumulative cell continuity=0
WQ Output face conc=0
WQ Output face dconc_dx=0
WQ Output face courant=0
WQ Output face peclet=0
WQ Output face adv mass=0
WQ Output face disp mass=0
WQ Output cell mass=0
WQ Output cell source sink temp=0
WQ Output nsm pathways=0
WQ Output nsm derived pathways=0
WQ Output MaxMinRange=-1
WQ Daily Max Min Mean=-1
WQ Daily Range=0
WQ Daily Time=0
WQ Create Restart=0
WQ Fixed Restart=0
WQ System Summary=0
WQ Write To DSS=0
WQ Use Fixed Temperature=0
Sorting and Armoring Iterations= 10
XS Update Threshold= 0.02
Bed Roughness Predictor= 0
Hydraulics Update Threshold= 0.02
Energy Slope Method= 1
Volume Change Method= 1
Sediment Retention Method= 0
XS Weighting Method= 0
Number of US Weighted Cross Sections= 1
Number of DS Weighted Cross Sections= 1
Upstream XS Weight=0
Main XS Weight=1
Downstream XS Weight=0
Number of DS XS's Weighted with US Boundary= 1
Upstream Boundary Weight= 1
Weight of XSs Associated with US Boundary= 0
Number of US XS's Weighted with DS Boundary= 1
Downstream Boundary Weight= 0.5
Weight of XSs Associated with DS Boundary= 0.5
Percentile Method= 0
Sediment Output Level= 3
Mass or Volume Output= 0
Output Increment Type= 1
Profile and TS Output Increment= 1
XS Output Flag= 0
XS Output Increment= 10
Write Gradation File= 0
Read Gradation Hotstart= 0
Write HDF5 File= 1
Write Binary Output= 1
Write DSS Sediment File= 0
SV Curve= 0
Specific Gage Flag= 0

--- SmithFork2019.f04 (steady flow) ---

Flow Title=2019 Smith Fork Flows
Program Version=5.07
Number of Profiles= 9
Profile Names=100-year,Floodway,2-year,5-year,10-year,25-year,50-year,200-year,500-year
River Rch & RM=Smith Fork River,Reach-1         ,26257
   36044   36044   11168   17236   21706   27281   31540   40653   47288
River Rch & RM=Smith Fork River,Reach-1         ,11972
   36990   36990   11461   17688   22275   27997   32368   41720   48529
Boundary for River Rch & Prof#=Smith Fork River,Reach-1         , 1
Up Type= 0
Dn Type= 3
Dn Slope=0.00024
Boundary for River Rch & Prof#=Smith Fork River,Reach-1         , 2
Up Type= 0
Dn Type= 3
Dn Slope=0.00024
DSS Import GetInterval= 0
DSS Import GetPeak= 0
DSS Import FillOption= 0

--- SmithFork2019.f06 (steady flow) ---

Flow Title=2019 Caney Flow Normal Depth
Program Version=5.07
Number of Profiles= 2
Profile Names=100-year,Floodway
River Rch & RM=Caney Fork,1               ,26.95
   30000   30000
River Rch & RM=Caney Fork,1               ,20.56
   49966   49966
River Rch & RM=Caney Fork,1               ,16.05
   75887   75887
River Rch & RM=Caney Fork,1               ,11.92
   85646   85646
River Rch & RM=Caney Fork,1               ,0.16
   93534   93534
Boundary for River Rch & Prof#=Caney Fork,1               , 1
Up Type= 0
Dn Type= 3
Dn Slope=0.00035
Boundary for River Rch & Prof#=Caney Fork,1               , 2
Up Type= 0
Dn Type= 3
Dn Slope=0.00035
Observed WS=Caney Fork      ,1               ,14.91   ,0.05,492,
Observed WS=Caney Fork      ,1               ,11.4    ,0,491.3,
Observed WS=Caney Fork      ,1               ,7.7     ,0,488,
Observed WS=Caney Fork      ,1               ,3.37    ,0,486.3,
DSS Import GetInterval= 0
DSS Import GetPeak= 0
DSS Import FillOption= 0

--- SmithFork2019.g07 (geometry) ---

Geom Title=Existing Conditions 2019 Smith Fork
Program Version=5.07

River Reach=Smith Fork River,Reach-1
Reach XY= 30
      2001306.61       643804.16      2002438.69       645758.88
      2002875.81        645646.1      2004046.59       644941.27
      2004359.98       644633.87      2004573.73        644116.3
      2004825.25       643957.54      2006080.06       644342.52
      2006630.58       645118.15      2006694.56       645768.01
      2007160.99       646855.98      2006108.02       648597.39
      2006086.44       648808.57      2006370.65       649488.49
      2006860.36       650186.42      2007019.68       651003.83
      2007554.54       651585.51      2007347.97       652034.15
      2006408.92       652692.74       2005962.2       653622.08
       2006408.2       654247.54      2006899.99       654445.54
      2007581.18       654371.52      2008490.35       653917.24
      2009137.22       655015.27       2008959.7        655286.7
      2008174.07       655705.83      2007095.34       655875.54
      2006936.14       656556.53      2007041.22        657534.7

Type RM Length L Ch R = 1 ,26257   ,911.8,915.6,914.1
BEGIN DESCRIPTION:
Smith Fork River 51.0
END DESCRIPTION:
XS GIS Cut Line= 3
      1999623.89       644830.742001743.37231625643555.712142098
      2001978.94       643291.12
#Sta/Elev= 30
       0   601.3   109.7  572.94   126.1  565.57   198.6  559.49   220.8  554.48
   233.5  556.84   252.9  556.36   280.9  550.23   499.5   533.7   875.5  520.25
  1058.8  520.03  1362.7  506.62  1835.3   503.5  1900.4  498.82  1911.2  494.35
  1925.8  483.97  2045.4  484.06  2051.2  495.18  2375.1  507.92  2428.6  516.06
  2477.7  531.72  2507.8  532.38  2532.6  537.07  2547.5  542.38  2605.2  544.97
  2632.4  556.24  2647.9  570.59  2677.5  586.22  2753.9  610.75  2827.7  629.53
#Mann= 3 , 0 , 0
       0     .16       0  1911.2     .06       0  2051.2     .16       0
Bank Sta=1911.2,2051.2
XS Rating Curve= 0 ,0
Exp/Cntr=0.3,0.1

Type RM Length L Ch R = 1 ,25342   ,858.1,862,859.4
BEGIN DESCRIPTION:
Smith Fork River 50.0
END DESCRIPTION:
XS GIS Cut Line= 5
1996442.58039452645418.2461622541998389.59049417644852.824888781
2000376.62728342645424.3177706452002009.89569213644463.661398372
      2002350.86       644466.43
#Sta/Elev= 30
       0  978.31   170.8   964.9   246.3  944.32   360.8   893.1   718.5  822.52
  1040.3  725.82  1191.2  689.75  1313.6   684.8    1684  793.03  1998.7  841.26
    2091  843.62  2198.6  825.44  2547.2  732.95  2695.5  706.61  3206.1  670.65
  3360.5  640.98  3624.1  636.81  3738.6  619.47  4114.3  527.22  4440.1  511.43
  5626.4  496.83  5643.8  483.19  5742.4  483.19  5761.6  495.99  5954.1  500.83
    5986  521.47  6009.1  522.94  6064.1  561.72  6097.4  567.73  6330.9  578.02
#Mann= 3 , 0 , 0
       0     .16       0  5626.4     .06       0  5761.6     .16       0
Bank Sta=5626.4,5761.6
XS Rating Curve= 0 ,0
Exp/Cntr=0.3,0.1

Type RM Length L Ch R = 1 ,24480   ,582.1,506.2,451.1
BEGIN DESCRIPTION:
Smith Fork River 49.0
END DESCRIPTION:
XS GIS Cut Line= 5
  1998965.900086648866.3615901662001314.66968146647312.145397667
2001401.03152972645793.3493385662002367.13254763645251.268924863
      2002373.97       644675.39
#Sta/Elev= 30
       0 1002.63   160.3  995.94   360.2  952.51   483.4  941.02   897.1  981.21
  1320.1  963.31  1769.5  996.43  1949.4  991.53  2078.3  970.61  2334.9  904.88
  2597.6  902.28  2770.4  888.49  2848.3  863.81  3068.7  828.04  3241.6   785.9
  3359.1  798.56  3554.4  800.34  3761.5   782.7  3950.8  726.97  4035.2  683.82
  4278.1  520.72  4338.4  509.08  5188.6  495.56  5198.3  494.79    5204  482.47
  5310.1   482.5  5319.3493.5689  5378.9   513.4  5737.9  514.47  6021.4  548.94
#Mann= 3 , 0 , 0
       0     .16       0  5188.6     .05       0  5319.3     .16       0
Bank Sta=5188.6,5319.3
XS Rating Curve= 0 ,0
Exp/Cntr=0.3,0.1

Type RM Length L Ch R = 1 ,23973   ,634.3,548.9,497.9
BEGIN DESCRIPTION:
Smith Fork River 48.0
END DESCRIPTION:
XS GIS Cut Line= 4
 2002259.0570305646110.2680811052002405.12971224645894.469827772
2002541.53169569645519.865119778      2002416.56       644663.25
#Sta/Elev= 30
       0  688.57    16.1  679.77    39.1  671.81    51.2  663.82    59.3  655.87
    78.4  642.79   111.5  613.01   120.6  592.54   123.6  589.27   211.2  540.07
   241.4  514.92   247.4  512.44   288.9  509.57   310.2  494.09   321.5  489.75
   334.1  482.06   424.6  482.06   437.9  489.51   467.1  493.07   480.4  491.58
     523  495.95   623.8  498.44   661.6  502.07   749.2  501.16  1098.3  508.66
    1260   516.2  1278.3  515.23  1348.9  523.43  1457.3  540.95  1524.9  547.97
#Mann= 3 , 0 , 0
       0     .16       0   321.5     .05       0   437.9     .16       0
Bank Sta=321.5,437.9
XS Rating Curve= 0 ,0
Exp/Cntr=0.3,0.1

Type RM Length L Ch R = 1 ,23424   ,384.2,380.2,377.9
BEGIN DESCRIPTION:
Smith Fork River 47.0
END DESCRIPTION:
XS GIS Cut Line= 3
      2003049.51       646087.38 2003042.7423326645713.143399559
        2002447.       644724.12
#Sta/Elev= 30
       0  655.38      57  646.88     127  627.67     222  595.49   239.5  585.81
   264.5  577.15   324.6  550.49   329.6   545.6   337.1  532.93   344.6  525.75
   349.6  511.82   352.1  507.72   403.8   507.3   413.6  504.43   421.3  497.17
   434.7  484.84   444.4  481.69   535.6  481.74   541.1  482.72   550.2  493.27
   564.3  492.55   569.8494.6333   578.9  499.49   701.4  502.37  1104.2  503.88
    1235  511.84  1371.6  516.01  1384.4  520.97  1475.5  531.82  1528.9  540.88
#Mann= 3 , 0 , 0
       0     .16       0   421.3     .05       0   569.8     .16       0
Bank Sta=421.3,569.8
XS Rating Curve= 0 ,0
Exp/Cntr=0.3,0.1

Type RM Length L Ch R = 1 ,23044   ,533.8,555.4,528.7
BEGIN DESCRIPTION:
Smith Fork River 46.0
END DESCRIPTION:
XS GIS Cut Line= 3
      2003481.63       645892.622003384.86701414645535.377014144
2002669.63574033644434.672555801
#Sta/Elev= 30
       0   558.2    93.6  554.09   165.5  545.15   206.9  538.69   227.7  532.76
   279.5  523.43     295  512.76   326.1  513.74   344.1  512.21     382  496.47
   408.3  495.89   426.7  493.84     443  483.07   450.6  481.44   550.5  481.44
   553.2   483.4   560.9   495.7   569.9  498.86     593     497   683.3  499.74
   876.3  499.12   984.3  501.88  1309.3  504.32    1357  509.71  1371.8  513.55
  1404.7   513.7  1420.6  520.24  1523.2  544.91  1637.2  555.49  1682.8  565.24
#Mann= 3 , 0 , 0
       0     .16       0   408.3     .05       0   560.9     .16       0
Bank Sta=408.3,560.9
XS Rating Curve= 0 ,0
Exp/Cntr=0.3,0.1

Type RM Length L Ch R = 1 ,22489   ,616.6,596.8,587.5
BEGIN DESCRIPTION:
Smith Fork River 45.0
END DESCRIPTION:
XS GIS Cut Line= 3
      2004303.76       646156.032003830.16574033645239.690206851
2002967.69892486644062.692779004
#Sta/Elev= 30
       0  631.59    65.5  612.32     133  597.46   147.1  590.35   189.9  587.89
   245.6  571.77   273.7  569.77   307.5  561.76   372.2  557.35   488.2  536.15
   515.7  533.82   586.5  538.41     670  537.69   909.3   526.6   987.3  515.14
  1058.6  493.62  1078.3  490.97  1098.8  481.09  1181.4  481.25  1217.9 493.146
  1241.1  498.04  1997.4  501.46  2056.7  504.33  2078.2  508.44  2223.9  513.31
  2262.4  520.62  2273.5  515.67  2292.8  524.17  2406.7  550.72  2490.7  562.98
#Mann= 3 , 0 , 0
       0     .16       0  1058.6     .05       0  1217.9     .16       0
Bank Sta=1058.6,1217.9
XS Rating Curve= 0 ,0
Exp/Cntr=0.3,0.1

Type RM Length L Ch R = 1 ,21892   ,418.1,346.8,318.5
BEGIN DESCRIPTION:
Smith Fork River 44.0
END DESCRIPTION:
XS GIS Cut Line= 4
      2005226.67       645490.482004499.78168752645036.204028289
2003979.93813347644540.257138704      2003238.22       643926.84
#Sta/Elev= 30
       0   570.5    53.2  570.15   150.5  565.25   395.2  542.84   506.3  529.25
   682.3   514.5   894.6   508.2    1120  512.73  1131.1  509.62 1147.98495.8334
  1169.8  480.69  1270.3  480.83  1273.8  481.86  1283.1   492.9  1290.3495.5524
  1386.8   497.6    1580  496.32  1702.2  498.39  1911.8  498.22  2149.7  501.51
  2167.5  506.27  2192.3  505.22    2207  507.95  2268.7  530.18    2361  545.82
  2439.7  543.99  2509.1  547.06  2516.9  545.72  2524.7  551.66  2538.1  555.07
#Mann= 3 , 0 , 0
       0     .16       0 1147.98     .05       0  1290.3     .16       0
Bank Sta=1147.98,1290.3
XS Rating Curve= 0 ,0
Exp/Cntr=0.3,0.1

Type RM Length L Ch R = 1 ,21545   ,491.7,577.1,624.3
BEGIN DESCRIPTION:
Smith Fork River 43.0
END DESCRIPTION:
XS GIS Cut Line= 4
      2005064.08        645271.92004720.35849481644602.533821437
2004071.85302186644371.7465099742002651.76600174642751.367425368
#Sta/Elev= 30
       0  562.49    91.6  555.13   291.2  526.05     398  514.82   585.6  509.66
   875.9  514.17     929   512.1   974.1  496.23   976.7  490.95   979.4  480.47
  1080.2  480.56  1114.7  496.97    1794  497.78  1947.9  503.03  2031.9  534.53
  2090.8  549.94  2207.4  557.84  2308.3  558.87  2397.1   566.6  2514.7  580.72
  2715.8   611.5  3058.2  688.39  3191.2  726.99  3242.9   748.4  3309.2   767.6
  3371.2  792.37  3443.9  813.12  3516.9  822.87  3546.8  821.37  3595.4   812.7
#Mann= 3 , 0 , 0
       0     .16       0   974.1     .05       0  1114.7     .16       0
Bank Sta=974.1,1114.7
XS Rating Curve= 0 ,0
Exp/Cntr=0.3,0.1

Type RM Length L Ch R = 1 ,20968   ,497.8,598.1,667.6
BEGIN DESCRIPTION:
Smith Fork River 42.0
END DESCRIPTION:
XS GIS Cut Line= 5
2005180.38020685645183.187237348  2004886.831699644331.916725001
2004574.47086011643795.8187343642005387.09943123643259.763021326
2006516.50845819642540.095525695
#Sta/Elev= 30
       0  556.77   370.5  514.49   833.3  512.22    1176  494.31  1194.3   487.5
  1318.1  480.09  1344.2  488.11  1356.5  495.62  1569.7  504.06  1718.1  574.91
  1721.5  581.64  1724.9  602.01  1735.7  627.86  1748.1   644.7  1757.3  667.03
    1775  679.92  1816.9  679.17  1861.9  690.06  1915.8  739.32  1930.7  745.88
  2221.1  836.96  2327.6  856.94  2459.3   903.1  2535.6  901.42  2844.9  822.31
  2971.1  819.65  3107.4  845.71  3208.8  890.47  3409.8  937.76  3833.6   975.9
#Mann= 3 , 0 , 0
       0     .16       0  1194.3     .05       0  1344.2     .16       0
Bank Sta=1194.3,1344.2
XS Rating Curve= 0 ,0
Exp/Cntr=0.3,0.1

Type RM Length L Ch R = 1 ,20370   ,495.6,505.7,510.6
BEGIN DESCRIPTION:
Smith Fork River 41.0
END DESCRIPTION:
XS GIS Cut Line= 4
2005250.44169569645189.314896574 2005165.6401938644524.937990637
2005298.14765105643947.518089281       2005216.2       643628.63
#Sta/Elev= 30
       0  556.35    82.1  549.29   281.2  524.33   326.6   522.5   353.4  519.04
   497.9  512.38   684.7  511.85   792.4  502.59  1066.9  493.04    1072  492.27
  1076.3  488.79  1084.8  479.47  1200.3  479.47  1215.6491.2052  1223.3  496.64
  1246.4  498.28  1264.4  515.52    1298  536.63  1308.4  555.22    1316  578.99
  1322.7  592.94  1341.8  625.35  1363.7  643.25  1419.2  681.45  1434.8  689.36
  1473.5  714.87  1525.1  737.98  1535.4  745.57  1563.8  761.08  1591.4  769.16
#Mann= 3 , 0 , 0
       0     .16       0  1076.3     .05       0  1215.6     .16       0
Bank Sta=1076.3,1215.6
XS Rating Curve= 0 ,0
Exp/Cntr=0.3,0.1

Type RM Length L Ch R = 1 ,19864   ,405.2,443.7,460.9
BEGIN DESCRIPTION:
Smith Fork River 40.0
END DESCRIPTION:
XS GIS Cut Line= 3
      2005423.14       645229.25 2005794.5829695644082.833407734
2005773.80403646643902.482340773
#Sta/Elev= 30
       0  558.54   101.1  554.71   232.7  554.91   306.3  549.06   382.5  536.85
   456.1  517.68   490.2  503.67   519.1  503.38   540.2   507.4   592.7  500.53
   950.1  495.38   984.3  494.13  1014.1  487.92  1031.6  478.88  1143.1  478.93
  1149.5  488.09    1163  496.54  1194.5  498.05  1207.3  511.42  1227.7  525.18
  1232.7  531.73  1265.4  557.76    1273  556.37  1283.1  531.59  1288.1   529.4
  1291.3   533.5  1300.3  558.23  1308.2   575.4  1329.6  606.05  1386.6  642.08
#Mann= 3 , 0 , 0
       0     .16       0  1014.1     .05       0  1149.5     .16       0
Bank Sta=1014.1,1149.5
XS Rating Curve= 0 ,0
Exp/Cntr=0.3,0.1

Type RM Length L Ch R = 1 ,19421   ,300.7,317.2,326.8
BEGIN DESCRIPTION:
Smith Fork River 39.0
END DESCRIPTION:
XS GIS Cut Line= 3
2005541.73085193645192.218089281 2006248.5729695644265.586600442
      2006202.16       644030.29
#Sta/Elev= 30
       0  556.58   137.5  553.44     213  549.09   272.7  543.08   310.5  537.15
   402.5  505.66   416.1   505.9   452.5  500.65   873.6  494.87   896.6  491.69
   906.6  487.25   917.3  483.45   923.6  478.34  1014.8  478.34    1025  483.61
  1039.3  484.43  1045.9487.4427  1058.9  495.69  1068.2  498.65  1090.2  498.71
  1170.8  508.55  1184.4  507.45  1198.8  513.49  1214.6  516.51  1229.4  527.63
  1252.5  535.97  1280.1   549.7  1325.1   560.4  1356.8  570.04  1405.3  577.93
#Mann= 3 , 0 , 0
       0     .16       0   906.6     .05       0  1045.9     .16       0
Bank Sta=906.6,1045.9
XS Rating Curve= 0 ,0
Exp/Cntr=0.3,0.1

Type RM Length L Ch R = 1 ,19103   ,611.8,638.1,652.7
BEGIN DESCRIPTION:
Smith Fork River 38.0
END DESCRIPTION:
XS GIS Cut Line= 3
2005729.78596354 645237.219371272006565.85743602 644436.94937127
      2006757.48       643613.62
#Sta/Elev= 30
       0     543   132.8  527.18   147.3  521.65     187  515.39   303.5  502.73
   396.9  498.75     777  494.53   807.1  486.92   812.5  480.13   819.2  477.91
     876  480.51     892  477.97   947.2  477.97   949.9  479.26   952.1  485.39
   953.8   489.3   962.7  493.22   996.9  499.35    1178  499.93  1194.9  497.08
  1220.6  503.09  1264.2  506.51  1343.8  526.75  1356.6  532.97  1366.9  533.37
  1400.2  548.27  1472.1  570.44  1767.4  625.33  1885.4  655.53  2002.7  681.69
#Mann= 3 , 0 , 0
       0     .16       0   807.1     .05       0   952.1     .16       0
Bank Sta=807.1,952.1
XS Rating Curve= 0 ,0
Exp/Cntr=0.3,0.1

Type RM Length L Ch R = 1 ,18465   ,377.5,408.8,422.9
BEGIN DESCRIPTION:
Smith Fork River 37.0
END DESCRIPTION:
XS GIS Cut Line= 3
      2005910.01       645582.272007037.31487205644987.511927071
      2008110.79       644878.17
#Sta/Elev= 30
       0  571.46   140.3  563.83   233.5  554.21   313.4  535.25   422.9  500.51
   479.9  496.16   746.4  490.42   750.8   489.1   756.5  477.16   869.5  477.29
   877.3  487.01   894.5493.9284   965.6  498.98  1287.2  504.52  1356.8  509.22
  1389.4  518.44  1439.7  542.99  1483.4  567.37  1565.3  624.41  1605.5  640.68
  1721.1  662.09  1832.3  672.52  1852.8  671.76    1897  681.46  1941.8   686.2
  1984.8  696.58  2026.2  700.65  2085.5  716.81  2248.8  752.44  2353.6  769.66
#Mann= 3 , 0 , 0
       0     .16       0   746.4     .05       0   894.5     .16       0
Bank Sta=746.4,894.5
XS Rating Curve= 0 ,0
Exp/Cntr=0.3,0.1

Type RM Length L Ch R = 1 ,18057   ,482.4,463.9,439.2
BEGIN DESCRIPTION:
Smith Fork River 36.0
END DESCRIPTION:
XS GIS Cut Line= 4
      2005830.14       645672.412006495.34224597645637.108140257
2007058.81253127645514.393837789      2007374.99645653.553192707
#Sta/Elev= 30
       0  567.92   219.2  565.74   366.9  556.19   532.2  531.23   597.3  516.19
   668.6  494.83   685.3  497.28   703.2  493.44   751.8  492.78   769.5  486.22
     780  478.56   805.6  482.97   823.5  480.71   840.9  482.92     867  478.19
   964.2  478.19   971.9  486.93     977  491.99   982.1  492.92  1202.1  497.25
  1305.9  504.72  1319.6  517.24  1394.2  553.45  1482.7  612.99  1497.1  623.65
  1513.5  644.78  1530.2   655.3  1537.7  664.51    1568  691.02  1588.3  705.23
#Mann= 3 , 0 , 0
       0     .16       0   769.5     .05       0   971.9     .16       0
Bank Sta=769.5,971.9
XS Rating Curve= 0 ,0
Exp/Cntr=0.3,0.1

Type RM Length L Ch R = 1 ,17593   ,416.6,415.9,412.3
BEGIN DESCRIPTION:
Smith Fork River 35.0
END DESCRIPTION:
XS GIS Cut Line= 5
2005749.76297523646174.3817104082006043.29086017646121.633992624
2006559.68266785646173.2783225812007115.21488022645872.788949391
2007395.98084376 645814.41341591
#Sta/Elev= 30
       0  565.28    52.6  552.73   174.6   538.2   192.3  532.66   286.3  515.96
   329.2  509.38   399.5  503.76   630.7   497.1    1024  499.04  1032.5  497.36
    1044  490.34  1049.6  484.44  1060.9  478.16  1163.3  478.45  1180.3  490.99
  1184.1  491.55  1329.8  490.39  1367.9  491.55  1396.2  497.33  1421.9  497.69
  1480.8  533.42  1511.5   554.6  1523.8  565.61    1545  578.36    1560  605.05
  1572.5  618.14  1585.5   639.2  1621.3  668.34  1697.9  705.79  1735.6  719.63
#Mann= 3 , 0 , 0
       0     .16       0    1044     .05       0  1184.1     .16       0
Bank Sta=1044,1184.1
XS Rating Curve= 0 ,0
Exp/Cntr=0.3,0.1

Type RM Length L Ch R = 1 ,17177   ,708.7,809.7,854.7
BEGIN DESCRIPTION:
Smith Fork River 34.0
END DESCRIPTION:
XS GIS Cut Line= 5
2005784.53106696646596.3504415012005968.83980056646587.642476803
2006587.25713437646642.0442534122007188.31956995646298.103630938
2007483.04979315646031.808312485
#Sta/Elev= 30
       0  582.23    58.9  563.06   154.7   516.1   167.2  515.15   184.7  508.17
   257.5  500.86   332.6  497.51   445.7  497.03  1071.7  498.34  1161.7  495.26
  1210.7  491.44  1214.6  488.32  1231.5  478.16  1360.4  478.16  1374.8  487.98
  1412.7  491.19  1423.8  495.93    1444  494.75  1455.5  503.19  1473.1  509.61
  1492.9   524.7  1505.6  562.12  1510.9  566.08  1525.1  567.96    1546  576.61
  1598.8  590.19  1702.1  625.73  1759.2  639.62    1829  663.31    1895  679.63
#Mann= 3 , 0 , 0
       0     .16       0  1214.6     .05       0  1374.8     .16       0
Bank Sta=1214.6,1374.8
XS Rating Curve= 0 ,0
Exp/Cntr=0.3,0.1

Type RM Length L Ch R = 1 ,16367   ,463.5,465.7,467.2
BEGIN DESCRIPTION:
Smith Fork River 33.0
END DESCRIPTION:
XS GIS Cut Line= 4
      2005843.04       646921.212006575.00181591 646911.66125938
 2007204.4429695647223.251695691       2007622.7        647189.9
#Sta/Elev= 30
       0  571.27      21   560.9    38.9  555.35      71  530.31   118.5  507.61
   128.5  507.62   148.5  501.46   173.5  498.14   303.6  495.41  1033.4  498.46
  1131.5  494.46  1165.1  485.33  1188.5   484.5    1194  478.12  1286.1  478.12
  1291.7  481.97  1294.5  486.43    1300  491.96  1310.7  496.22  1327.9   516.1
  1394.1  536.77  1400.5   541.7  1425.6  544.76    1444  543.48  1476.6  554.63
  1549.4  573.23  1599.5  582.37    1727  613.13  1792.6  623.37    1854   628.3
#Mann= 3 , 0 , 0
       0     .16       0  1188.5     .05       0  1294.5     .16       0
Bank Sta=1188.5,1294.5
XS Rating Curve= 0 ,0
Exp/Cntr=0.3,0.1

Type RM Length L Ch R = 1 ,15901   ,620.2,627.5,633.3
BEGIN DESCRIPTION:
Smith Fork River 32.0
END DESCRIPTION:
XS GIS Cut Line= 4
      2005873.26       647319.972006375.85289105 647313.02293872
2007019.13594718647658.339991824      2007467.47       647433.93
#Sta/Elev= 30
       0   568.3    25.8   560.4    35.8  550.05    53.3  536.05   108.3  506.58
   120.8  506.61   130.8  499.87   143.3   497.4   275.8  494.34   308.3  496.18
   728.3  497.93   880.8  494.06   906.4  488.46   923.4  487.46   926.2  486.39
   931.9  478.12  1041.5  478.12  1042.6  478.33  1048.2  487.98  1082.3  500.47
    1153  514.11  1238.3  523.44  1263.4  523.86  1333.6  531.61  1372.5  533.22
  1397.6  537.28  1447.9  538.89  1495.7  549.49    1557  556.37  1734.1  589.45
#Mann= 3 , 0 , 0
       0     .16       0   923.4     .05       0  1048.2     .16       0
Bank Sta=923.4,1048.2
XS Rating Curve= 0 ,0
Exp/Cntr=0.3,0.1

Type RM Length L Ch R = 1 ,15274   ,360.4,357.6,352.9
BEGIN DESCRIPTION:
Smith Fork River 31.0
END DESCRIPTION:
XS GIS Cut Line= 4
      2005853.08       647849.452006247.17204729647922.725031762
2006824.75998365648305.410198675      2007436.41       648392.37
#Sta/Elev= 30
       0  569.78    23.9  561.92    82.4  533.75     118  519.12   153.9  505.77
   191.7  495.36   255.3  491.12     543  495.72   580.9  494.03   604.8  488.28
     625  487.56   627.8  486.49     634  477.97     742  477.97     757  488.74
   784.7  496.93     823  496.39  1050.9  504.01  1166.2  510.79  1229.4  517.15
  1330.4  534.98  1385.9  549.81  1406.1  549.99  1423.8  555.43  1466.5  562.67
    1497  571.84  1561.8   584.8  1605.6   599.7  1683.9  616.56  1711.5  624.56
#Mann= 3 , 0 , 0
       0     .16       0     625     .05       0     757     .16       0
Bank Sta=625,757
XS Rating Curve= 0 ,0
Exp/Cntr=0.3,0.1

Type RM Length L Ch R = 1 ,14916   ,461.2,416.1,363.7
BEGIN DESCRIPTION:
Smith Fork River 30.0
END DESCRIPTION:
XS GIS Cut Line= 4
      2005739.19       648231.512006020.44865591 648210.72501541
2006569.48764287 648547.47062873      2007169.89       648588.84
#Sta/Elev= 30
       0  589.73    17.4  589.37    37.5  585.83      50  577.66    65.1  574.79
    97.6  554.02   195.4  517.94     226  503.97   245.5  497.59     282  492.86
   403.6  492.99   468.1  491.12   495.3  487.83   506.1   484.9   510.9  478.97
     515  478.02   625.6  477.88   632.3   486.9   636.1489.6084   661.7  495.08
   693.9   493.6     779  493.91  1013.4  498.02  1073.8  500.91  1165.2  508.44
  1331.7  526.07  1446.9  549.78  1459.4  554.58    1482  554.96  1527.9  568.49
#Mann= 3 , 0 , 0
       0     .16       0   495.3     .05       0   636.1     .16       0
Bank Sta=495.3,636.1
XS Rating Curve= 0 ,0
Exp/Cntr=0.3,0.1

Type RM Length L Ch R = 1 ,14500   ,538.2,504.2,472.6
BEGIN DESCRIPTION:
Smith Fork River 29.0
END DESCRIPTION:
XS GIS Cut Line= 3
      2005745.83       648727.48      2006074.79       648722.09
      2007139.47        648692.3
#Sta/Elev= 30
       0  594.81    13.2  592.86    33.2  578.46    68.2  561.53   108.6  549.36
   118.3   540.3   123.3  537.86   147.9   529.3   195.8  516.76   213.3  509.39
   219.8  505.76   230.8  493.41   248.3   490.3   258.6  484.77   268.3  477.87
   270.8  477.78   393.3  477.78   395.8  478.29   398.3  485.01   400.8  487.27
   413.3  487.83   433.3  494.97   511.8   492.7   600.9  492.78   861.7  496.92
   987.8  502.45  1223.6  529.77  1354.2  550.97  1373.7  557.31  1394.1  557.69
#Mann= 3 , 0 , 0
       0     .16       0   258.6     .05       0   398.3     .16       0
Bank Sta=258.6,398.3
XS Rating Curve= 0 ,0
Exp/Cntr=0.3,0.1

Type RM Length L Ch R = 1 ,13996   ,470.5,469.1,443.1
BEGIN DESCRIPTION:
Smith Fork River 28.0
END DESCRIPTION:
XS GIS Cut Line= 3
2005858.15319271649382.7248965742006515.13381326649054.103837789
      2007224.63       648880.97
#Sta/Elev= 30
       0  619.75    13.6  613.92      29   603.6    51.3  603.66    68.1  600.98
   140.8  569.06   171.5  553.16   219.1  541.56   244.2  541.88   269.4  536.41
   316.9  509.06   321.1  504.24   329.4  489.62   333.7  478.19     335  477.78
   445.5  477.78   451.1  480.03   462.2  489.31   467.7490.9478   495.8  489.58
   965.1  498.77  1024.5  505.22  1104.1   520.8  1148.4  526.91  1268.4  532.91
  1327.2  539.55  1412.9  556.36  1428.3  561.63  1451.5  562.47  1464.9  568.02
#Mann= 3 , 0 , 0
       0     .16       0   329.4     .05       0   467.7     .16       0
Bank Sta=329.4,467.7
XS Rating Curve= 0 ,0
Exp/Cntr=0.3,0.1

Type RM Length L Ch R = 1 ,13527   ,454.4,471.1,454.9
BEGIN DESCRIPTION:
Smith Fork River 27.0
END DESCRIPTION:
XS GIS Cut Line= 3
      2006241.82       649752.982006785.65615403649336.755971711
      2007182.05       649106.15
#Sta/Elev= 30
       0  555.35    33.8  544.88    43.8  540.23    78.3  528.62   115.3  513.33
   128.3  509.76   141.3  504.52   162.2  499.04   172.9  492.73   176.4  488.42
   185.4  483.69   188.9  479.32   191.7  477.78   327.1  477.78   333.4  480.63
   339.7  485.34   345.7  487.69   364.4489.3521   424.3   492.4   613.6  493.01
   670.4  495.11   723.1  503.14   821.8  525.56   856.4  529.96   992.5  535.36
  1010.7   537.1  1032.1  536.87  1041.6  535.57  1073.5  535.68  1143.4  542.26
#Mann= 3 , 0 , 0
       0     .16       0   176.4     .05       0   364.4     .16       0
Bank Sta=176.4,364.4
XS Rating Curve= 0 ,0
Exp/Cntr=0.3,0.1

Type RM Length L Ch R = 1 ,13056   ,1073.3,1083.9,1094.7
BEGIN DESCRIPTION:
Smith Fork River 26.0
END DESCRIPTION:
XS GIS Cut Line= 3
2006176.72276265650370.2653184532006930.91828796649798.367245524
      2007170.13       649244.31
#Sta/Elev= 30
       0  622.09      72  607.36    87.7  599.19    99.7   587.8   112.8  587.22
   119.4  583.24   165.8  584.46   194.3  571.37   219.4  565.85   238.3   554.6
   294.7  537.49     301  532.55   366.9   507.6   410.8  504.73   445.9  498.05
   500.5  495.48   550.1  489.99   595.8  489.41   601.1  486.49   604.7  478.47
   606.5  477.82   740.2  477.78   745.7  484.61   755.9  490.42   781.4  488.82
   870.6  492.11   947.4  508.53  1072.3  513.46  1344.6  531.71    1550  538.04
#Mann= 3 , 0 , 0
       0     .16       0   601.1     .05       0   745.7     .16       0
Bank Sta=601.1,745.7
XS Rating Curve= 0 ,0
Exp/Cntr=0.3,0.1

Type RM Length L Ch R = 1 ,11972   ,475.3,442.6,415.8
BEGIN DESCRIPTION:
Smith Fork River 24.0
END DESCRIPTION:
XS GIS Cut Line= 3
      2006406.99       651285.332007474.12359006 650753.30341591
      2007990.98       650730.71
#Sta/Elev= 30
       0  560.18    91.7  543.71   144.8  537.79   245.4  542.66   334.7  537.45
   359.9  533.55   380.9  527.97   457.7  503.27   504.8   495.6   588.2  487.19
   602.9  477.78   722.7  477.78   731.4  484.19   737.8  485.77   829.1  495.81
   920.5   493.7    1008  494.25  1293.5  507.39  1387.5  518.08  1417.6  523.63
  1442.6  533.82  1472.6  535.55    1514  552.65  1525.2  555.59  1600.2  593.14
  1605.4  594.41  1607.7  596.91  1649.8  619.45  1675.3  630.71  1709.8  649.02
#Mann= 3 , 0 , 0
       0     .16       0   588.2     .05       0   737.8     .16       0
Bank Sta=588.2,737.8
XS Rating Curve= 0 ,0
Exp/Cntr=0.3,0.1

Type RM Length L Ch R = 1 ,11529   ,317.3,387.2,434.2
BEGIN DESCRIPTION:
Smith Fork River 23.0
END DESCRIPTION:
XS GIS Cut Line= 4
      2006670.77       651400.652007212.27837547651409.363131671
2007599.99636906650992.117038672      2007863.65       651072.01
#Sta/Elev= 30
       0  537.88   200.8  522.41   358.3  508.59   543.9  501.09   570.9  497.51
   600.5  495.22   617.7  492.26   628.7  487.14   632.3     485     636  477.78
   753.5  477.78   757.2  478.81   768.1485.7243   771.9     487   856.4  493.17
   966.8  493.22  1000.3   494.5  1109.8  504.45  1128.5   507.7  1141.5  508.72
  1147.1  512.83    1152  514.59  1162.4  515.58  1175.2  514.91  1179.2  517.12
  1191.2   520.4  1214.7  529.48  1251.2  547.37  1323.5  570.52  1386.6  597.91
#Mann= 3 , 0 , 0
       0     .16       0   628.7     .05       0   768.1     .16       0
Bank Sta=628.7,768.1
XS Rating Curve= 0 ,0
Exp/Cntr=0.3,0.1

Type RM Length L Ch R = 1 ,11142   ,544,633,710.2
BEGIN DESCRIPTION:
Smith Fork River 22.0
END DESCRIPTION:
XS GIS Cut Line= 3
       2006634.3       651449.342007009.23907346651647.033374722
2008259.61487023651506.256824553
#Sta/Elev= 30
       0  539.62   358.7  505.08   687.9  499.04   801.1  492.47   848.9  491.93
     864  488.14   866.5  486.45     869   478.8   871.5  477.78  1009.9  477.78
  1025.6489.9312    1035  496.45  1060.2  498.92  1077.8  514.03  1168.4  563.21
  1198.6  581.65  1241.3  611.19  1304.8  658.85  1362.1  703.68  1367.1  711.57
  1450.1  768.51  1497.9  795.55  1525.6   808.3  1568.4  822.04    1581  828.46
  1598.6   842.9  1626.2  860.58  1652.2  871.55  1666.5  883.46  1682.1  891.45
#Mann= 3 , 0 , 0
       0     .16       0     864     .05       0  1025.6     .16       0
Bank Sta=864,1025.6
XS Rating Curve= 0 ,0
Exp/Cntr=0.3,0.1

Type RM Length L Ch R = 1 ,10509   ,285.3,293.5,293.2
BEGIN DESCRIPTION:
Smith Fork River 21.0
END DESCRIPTION:
XS GIS Cut Line= 4
      2006603.85       651479.762006900.30290943651704.905711862
2007341.68339865652222.917653776      2007735.88       652289.23
#Sta/Elev= 30
       0  540.65   368.1  505.38   534.9  499.75   619.2  493.67   796.6  490.16
   806.4  489.24     813  484.83   816.8  479.51   819.6  477.66   944.4  477.66
   946.3  478.33   950.9  483.98   960.1  490.68   965.8  496.88   994.8   499.3
  1002.5  506.85  1010.1  516.84  1019.9  521.53  1025.6  526.25  1029.5  526.83
  1033.1  530.48  1042.9  531.97  1049.2  534.93  1080.6  556.47  1090.7  561.18
  1126.2  572.47  1214.9  596.64  1304.4  611.93  1397.7  622.82  1452.5  624.85
#Mann= 3 , 0 , 0
       0     .16       0     813     .05       0   950.9     .16       0
Bank Sta=813,950.9
XS Rating Curve= 0 ,0
Exp/Cntr=0.5,0.3

Type RM Length L Ch R = 1 ,10215   ,232.8,230.9,230.5
XS GIS Cut Line= 3
2006552.05508104651678.1857254132007356.00270442652730.052634957
2007582.99105654652876.204377013
#Sta/Elev= 30
       0   527.5   118.6   516.6   139.2  516.88   229.7  511.49   460.3  491.47
   635.2  491.08   643.3  488.54   645.6  485.27   646.8  481.65   649.7  477.62
   808.3  477.62   811.6481.5073   814.6  486.19   835.9  491.17   882.3  491.99
   921.4  499.22   935.8  497.22   954.3  502.01   978.6  502.65  1126.1  518.56
    1167  518.95  1172.5  521.41  1182.7  521.14    1189  523.22  1201.3  523.92
  1280.3  523.05  1313.9  525.14    1497  543.09  1547.6  545.59  1593.9  550.24
#Mann= 3 , 0 , 0
       0     .16       0   646.8     .05       0   811.6     .16       0
#XS Ineff= 2 , 0
             401  511.69    1019          514.68
Permanent Ineff=
       F       F
Bank Sta=646.8,811.6
XS Rating Curve= 0 ,0
Exp/Cntr(USF)=0,0
Exp/Cntr=0.5,0.3

Type RM Length L Ch R = 3 ,10119   ,,,
Bridge Culvert--1,0,-1,-1, 0
Deck Dist Width WeirC Skew NumUp NumDn MinLoCord MaxHiCord MaxSubmerge Is_Ogee
80,39,2.6,0, 12, 12, , , 0.98, 0, 0,0,,
       0   86.09  152.22   196.2     481     481     939     939   947.6 1050.33
 1213.81 1552.34
  519.63  519.65  516.47  511.45     514   516.7   516.4   513.9  514.06  514.68
  520.16  536.26
                                           510.7   510.7
                
       0   86.09  152.22   196.2  481.69     539     539     997     997 1050.33
 1213.81 1552.34
  519.63  519.65  516.47  511.45   513.8   513.9   516.6   516.6   513.9  514.68
  520.16  536.26
                                                   510.6   510.6
                
Pier Skew, UpSta & Num, DnSta & Num=  ,506, 2 ,564, 2 , 0 , 0 , 0 ,,
       1       1
       0   510.7
       1       1
       0   510.7
Pier Skew, UpSta & Num, DnSta & Num=  ,535, 2 ,593, 2 , 0 , 0 , 0 ,,
       1       1
       0   510.7
       1       1
       0   510.7
Pier Skew, UpSta & Num, DnSta & Num=  ,565, 2 ,623, 2 , 0 , 0 , 0 ,,
       2       2
       0   510.7
       2       2
       0   510.7
Pier Skew, UpSta & Num, DnSta & Num=  ,646, 2 ,704, 2 , 0 , 0 , 0 ,,
       3       2
       0   510.7
       3       2
       0   510.7
Pier Skew, UpSta & Num, DnSta & Num=  ,743, 2 ,801, 2 , 0 , 0 , 0 ,,
       3       2
       0   510.7
       3       2
       0   510.7
Pier Skew, UpSta & Num, DnSta & Num=  ,827, 2 ,885, 2 , 0 , 0 , 0 ,,
       2       2
       0   510.7
       2       2
       0   510.7
Pier Skew, UpSta & Num, DnSta & Num=  ,857, 2 ,915, 2 , 0 , 0 , 0 ,,
       2       2
       0   510.7
       2       2
       0   510.7
Pier Skew, UpSta & Num, DnSta & Num=  ,887, 2 ,945, 2 , 0 , 0 , 0 ,,
       2       2
       0   510.7
       2       2
       0   510.7
Pier Skew, UpSta & Num, DnSta & Num=  ,917, 2 ,975, 2 , 0 , 0 , 0 ,,
       2       2
       0   510.7
       2       2
       0   510.7
BR Coef=-1 , 1 , 0 ,, 0 ,,,0.8,0,1.85,0,
WSPro=,,,, 1 ,,,, 0 ,,,, 0 ,,,,-1 ,-1 ,-1 , 0 , 0 , 0 , 0 , 0
BC Design=,, 0 ,, 0 ,,,,,,
BC Use User HTab Curves=0
BC User HTab FreeFlow(D)= 0

Type RM Length L Ch R = 1 ,9984    ,306,307.3,314.3
XS GIS Cut Line= 3
2006336.82059302651791.4230447522007166.74693455652845.384380654
2007407.13921972653011.423175955
#Sta/Elev= 30
       0  516.95   127.3  506.32   138.7  506.89   149.1  511.07   176.9  510.96
   208.7  505.58   242.1  503.73   258.2  496.72   278.6  494.07   324.9   493.2
   358.2  498.35   371.4  495.66   453.7  491.71   561.9  490.38   654.2  492.66
   657.8  492.09   663.1  487.46   666.9  480.06   670.1  477.62   813.3  477.62
   819.6  479.96   835.8  480.87   852.2  484.76   919.5  488.95   969.2   494.5
  1185.6   501.2  1243.5  504.34  1268.4  508.06  1334.2  510.32  1633.7  535.99
#Mann= 3 , 0 , 0
       0     .16       0   666.9     .05       0   819.6     .16       0
#XS Ineff= 2 , 0
           481.5     511  1054.5             511
Permanent Ineff=
       F       F
Bank Sta=666.9,819.6
XS Rating Curve= 0 ,0
Exp/Cntr(USF)=0,0
Exp/Cntr=0.5,0.3

Type RM Length L Ch R = 1 ,9677    ,535.4,492,454.3
BEGIN DESCRIPTION:
Smith Fork River 19.0
END DESCRIPTION:
XS GIS Cut Line= 5
2005400.14642294650091.0028410542005829.54480349 651035.88469842
2005912.72729782651737.0215324592006705.43105243652757.694246041
       2007298.8       653388.52
#Sta/Elev= 30
       0  880.09   120.1  847.53   245.1  801.31   353.9  773.78     399  768.11
   674.6  712.34   825.9  694.57   853.3  685.54   944.6  688.19   961.6  681.92
  1052.5  668.33  1304.2  620.71  1639.1  574.67    1888  535.97  2051.8  519.05
  2126.8  506.22  2161.8  505.99  2219.8  496.94  2248.3  498.29  2270.5  492.63
    2299  491.51    2704  492.53  2711.2  485.38    2720  477.16  2842.5  477.16
  2857.3  484.26    2925  480.27  3143.7  496.76  3578.8  514.26  3902.3  536.02
#Mann= 3 ,-1 , 0
       0     .16       0  2711.2     .05       0  2857.3     .16       0
Bank Sta=2711.2,2857.3
XS Rating Curve= 0 ,0
Exp/Cntr=0.3,0.1

Type RM Length L Ch R = 1 ,9185    ,682.7,658.1,638.3
BEGIN DESCRIPTION:
Smith Fork River 18.0
END DESCRIPTION:
XS GIS Cut Line= 5
2001570.85943719650118.1981343712004738.71693551651614.688161446
 2005882.4306268652753.4162906272006419.08254217653028.094255126
      2007187.86       653406.27
#Sta/Elev= 30
       0     869   157.3  898.94   310.5  915.91   484.8     906   708.6  874.71
   899.8  876.29   971.1  869.42    1621  906.08  1936.2  914.82  2049.6  910.16
  2190.6  888.61  2351.3  822.11  2881.8   676.8  3219.1   604.6  3476.3  564.53
  4195.5  490.31    4397   501.5  4677.3  503.49  4735.3  500.37  4784.6  487.88
  5313.1  492.22  5439.5  484.78  5447.9  476.12  5593.9  476.12  5610.8  482.79
  5701.6  483.06  5787.8  501.81  5845.7  506.57  5998.9  506.39  6577.1   535.8
#Mann= 3 ,-1 , 0
       0     .16       0  5439.5     .05       0  5610.8     .16       0
Bank Sta=5439.5,5610.8
XS Rating Curve= 0 ,0
Exp/Cntr=0.3,0.1

Type RM Length L Ch R = 1 ,8527    ,619.7,535.6,453.2
BEGIN DESCRIPTION:
Smith Fork River 17.0
END DESCRIPTION:
XS GIS Cut Line= 6
2001952.93682207655835.8718895862005082.57310762653850.061487213
2005417.20553577 653661.39941869 2005712.2178705653475.118377311
 2006352.5565741653624.896592266       2007187.9       653424.03
#Sta/Elev= 30
       0  989.78   110.9  983.45   481.5  923.99   827.4  949.06  1296.3  935.29
  1585.4  860.09  1711.2  847.35    1847  848.54  2035.4  906.73  2147.7  909.01
  2315.4  884.94  2464.7  814.62  2553.3  799.43  2663.1  812.77  2973.7  918.78
  3111.4  948.86  3239.3  946.47  3453.6  907.67  3711.1   904.2  4172.7  732.45
  4308.7  640.18  4376.7  568.28  4388.1  528.53  4439.5  503.29  4490.2  488.68
  4621.2  484.52  4626.5  475.79  4772.6  475.78  4793.2  482.82  5956.3  536.64
#Mann= 3 ,-1 , 0
       0     .16       0  4621.2     .05       0  4793.2     .16       0
Bank Sta=4621.2,4793.2
XS Rating Curve= 0 ,0
Exp/Cntr=0.3,0.1

Type RM Length L Ch R = 1 ,7992    ,522.3,491.6,466
BEGIN DESCRIPTION:
Smith Fork River 16.0
END DESCRIPTION:
XS GIS Cut Line= 3
2005940.97744874654178.3842551262006524.00125746653760.080651441
      2007099.12       653455.11
#Sta/Elev= 30
       0  656.85    36.6  642.53    45.6  634.89    78.1  614.29    86.9  610.13
   114.6  588.03   133.8  575.32   142.3  566.46   145.3  558.39   149.5  551.51
   160.2  523.27   163.8  515.58   166.9  511.42     171  508.25   185.3  507.28
   198.1  495.92   222.3  484.06   228.3  476.46   231.5   475.5   352.5   475.5
   366.5483.5367     434  483.93   506.9  492.03   643.9  493.72   702.3  496.12
     794  503.41  1011.4  509.26  1113.8  515.17  1283.6  529.86  1368.5  534.24
#Mann= 3 ,-1 , 0
       0     .16       0   222.3     .05       0   366.5     .16       0
Bank Sta=222.3,366.5
XS Rating Curve= 0 ,0
Exp/Cntr=0.3,0.1

Type RM Length L Ch R = 1 ,7500    ,482.1,427.8,400
BEGIN DESCRIPTION:
Smith Fork River 15.0
END DESCRIPTION:
XS GIS Cut Line= 3
      2006353.57       654594.36      2006535.64       654342.47
      2007108.98        653463.9
#Sta/Elev= 30
       0  634.41    21.1  630.47    60.6  616.62    81.9  603.26   101.7  594.03
   128.9  575.08   137.6  570.97     153   560.5   162.6  550.25   167.3  536.58
   173.3  515.93   176.9   510.8   180.7  501.92     190  496.14   217.8  493.16
   220.8  491.76   223.9  487.45   233.2  475.25   349.1  475.37   368.5 486.825
   411.8  489.21   536.6   482.9   647.2  492.81   780.8  492.64     873  495.13
   919.3  499.98  1021.5  505.21  1223.8  528.98  1297.5  533.62  1359.9   534.8
#Mann= 3 ,-1 , 0
       0     .16       0   223.9     .05       0   368.5     .16       0
Bank Sta=223.9,368.5
XS Rating Curve= 0 ,0
Exp/Cntr=0.3,0.1

Type RM Length L Ch R = 1 ,7072    ,604.1,562.3,531.6
BEGIN DESCRIPTION:
Smith Fork River 14.0
END DESCRIPTION:
XS GIS Cut Line= 3
      2006924.99       654775.032006954.74766286654166.723845057
 2007248.7448884653568.273826888
#Sta/Elev= 30
       0   702.4    44.7  675.86    54.7  667.07    94.8  640.02   172.4  582.82
   174.9  579.62   182.4  565.43   192.1  557.65   194.9  552.77   199.9   540.2
   204.9  515.27   207.4  508.36   209.9  504.87   214.9  500.77   229.9  499.12
   242.2  488.65   257.5  475.16   352.6  475.19   370.1  478.78   388.7486.9772
   442.7  486.47   510.3  482.39   540.5  484.27   610.5  492.62   777.6  491.87
   878.5  497.88   964.3  499.03  1017.2  504.15  1117.5  519.48  1275.8  536.92
#Mann= 3 ,-1 , 0
       0     .16       0   242.2     .05       0   388.7     .16       0
Bank Sta=242.2,388.7
XS Rating Curve= 0 ,0
Exp/Cntr=0.3,0.1

Type RM Length L Ch R = 1 ,6510    ,671,668.6,648.4
BEGIN DESCRIPTION:
Smith Fork River 13.0
END DESCRIPTION:
XS GIS Cut Line= 4
      2007449.67       654715.282007551.18531664654508.818929405
2007346.26033092654064.054514085      2007502.92       653353.08
#Sta/Elev= 30
       0  606.42    83.5  592.17   134.6  578.41   157.3  564.43   191.3  550.38
   203.3  540.62     206  535.43   206.8  531.17   208.8  512.65   210.5  508.04
   217.2  500.39     220  498.97   236.6  498.14   253.1     490   269.6  486.71
   272.4  482.06   275.1  475.99   277.9  474.81   423.8  474.81   434.8  476.41
   443.1  480.25   535.8  489.86   619.2  489.23   679.8  491.35   764.5  501.04
   846.4  504.53  1025.6  522.14  1153.1  532.31  1294.4  535.35  1447.8  535.95
#Mann= 3 ,-1 , 0
       0     .16       0   272.4     .05       0   443.1     .16       0
Bank Sta=272.4,443.1
XS Rating Curve= 0 ,0
Exp/Cntr=0.3,0.1

Type RM Length L Ch R = 1 ,5841    ,549.5,756.5,820
BEGIN DESCRIPTION:
Smith Fork River 12.0
END DESCRIPTION:
XS GIS Cut Line= 4
       2007560.3       654716.522008182.33714437654262.913572185
2007891.76856689653774.510533709      2007928.88       652833.88
#Sta/Elev= 30
       0  572.93   106.8  552.25   154.7  540.26   197.1  535.53   268.3  517.54
     282   517.5   286.2  507.62     288  506.38   311.7  498.21   369.8  492.16
   757.2  481.24   836.8  479.91   897.9  482.15   913.2   478.6   918.1  474.62
  1057.9  474.59  1060.8  478.35  1064.7  489.27  1072.4  491.52  1322.6  493.79
  1396.5  504.22  1467.7  518.35    1540  524.77  1730.1   533.2  1832.4  529.69
  1940.3  530.28  2020.3  537.12  2050.3  536.55  2067.9  540.76  2279.5  562.96
#Mann= 3 ,-1 , 0
       0     .16       0   913.2     .05       0  1060.8     .16       0
Bank Sta=913.2,1060.8
XS Rating Curve= 0 ,0
Exp/Cntr=0.3,0.1

Type RM Length L Ch R = 1 ,5085    ,1014.4,1097.9,1136.3
BEGIN DESCRIPTION:
Smith Fork River 11.0
END DESCRIPTION:
XS GIS Cut Line= 3
      2007601.23       654754.122008785.77196682654063.523391457
      2009906.34       652760.93
#Sta/Elev= 30
       0  556.66    55.4  543.72   110.4  534.54   223.2   520.1   275.4  510.18
   373.7   496.7   467.3  492.38     683  490.98   999.3  478.56  1102.9  484.36
  1117.4  482.31  1120.3  476.32  1123.2  474.38  1236.1  474.34  1253.3  482.66
    1265  492.87  1273.7  504.09  1278.1  506.22  1288.1  521.86    1291  522.79
  1583.1  515.09  1800.7  517.36  1827.1  515.05  1856.8  519.61  2084.3  525.76
  2341.9  515.99  2552.6  513.11  2944.1  520.21  3047.6  530.65  3089.4  540.31
#Mann= 3 ,-1 , 0
       0     .16       0  1117.4     .05       0  1253.3     .16       0
Bank Sta=1117.4,1253.3
XS Rating Curve= 0 ,0
Exp/Cntr=0.3,0.1

Type RM Length L Ch R = 1 ,3987    ,928.6,1035.1,1052.9
BEGIN DESCRIPTION:
Smith Fork River 8.0
END DESCRIPTION:
XS GIS Cut Line= 4
      2007691.13       654810.022009317.25518179655120.832143311
2009812.28194944 655489.520657162014177.42340144654483.630770206
#Sta/Elev= 30
       0  530.02     367  499.78   641.1  511.41  1311.3   487.4  1362.2  474.03
  1534.9  474.09  1568.3  486.99  1606.5  496.43  1633.2  556.55  1675.7  550.22
  1692.1  577.89  2158.6  751.45  2272.8  779.26  2451.7  756.28    2603  762.37
    2780  815.58  2946.8  885.16  2998.1  876.79  3149.5  803.95  3536.9  675.74
  4016.5   839.3    4098  853.15    4227  808.01  4475.8  753.45  4868.4  727.81
  5140.3  648.04  5250.6  632.37  5704.7  730.49  6420.7  778.38  6752.3  867.43
#Mann= 3 , 0 , 0
       0     .16       0  1311.3     .05       0  1568.3     .16       0
Bank Sta=1311.3,1568.3
XS Rating Curve= 0 ,0
Exp/Cntr=0.3,0.1
